--- SUGARRN.prj (project) ---

Proj Title=SUGARRN
Current Plan=p01
Default Exp/Contr=0,0
English Units
Geom File=g01
Flow File=f01
Plan File=p01
BEGIN DESCRIPTION:
---------- MODELED AS PART OF WVEMD CTP PROGRAM, 2023----------
Stream Name: Sugar Run
Flood Zone:  AFH
Wetzel County, WV
HEC-RAS Version: RAS 6.3
Vertical Datum: NAVD88
Projection: NAD 1983 StatePlane West Virginia S FIPS 4702 (US Feet)
Terrain: 1-meter West Virginia FEMA R3 South Central (collected 2018-2020)
Land Use: 2019 NLCD
Hydrologic Method:
WV SIR2010-5033 regression equations
Additional Model Notes:
None
END DESCRIPTION:
DSS File=dss
DSS Export Rating Curves= 0
DSS Export Rating Curve Sorted= 0
DSS Export Volume Flow Curves= 0
DXF OffsetX= 0
DXF OffsetY= 0
DXF ScaleX= 0
DXF ScaleY= 0

--- SUGARRN.p01 (plan) ---

Plan Title=Floodplain
Program Version=6.30
Short Identifier=Floodplain
Geom File=g01
Flow File=f01
Subcritical Flow
K Sum by GR= 0
Std Step Tol= 0.01
Critical Tol= 0.01
Num of Std Step Trials= 20
Max Error Tol= 0.3
Flow Tol Ratio= 0.001
Split Flow NTrial= 30
Split Flow Tol= 0.02
Split Flow Ratio= 0.02
Log Output Level= 0
Friction Slope Method= 1
Unsteady Friction Slope Method= 2
Unsteady Bridges Friction Slope Method= 1
Parabolic Critical Depth
Global Vel Dist= 0 , 0 , 0
Global Log Level= 0
CheckData=True
Encroach Param=-1 ,0,0, 0
Computation Interval=0.1SEC
Output Interval=1SEC
Instantaneous Interval=Max Profile
Mapping Interval=1HOUR
Computation Time Step Use Courant=        0
Computation Time Step Use Time Series=    0
Computation Time Step Count To Double=0
Computation Time Step Max Doubling=0
Computation Time Step Max Halving=0
Computation Time Step Residence Courant=0
Run HTab= 0
Run UNet= 0
Run Sediment= 0
Run PostProcess= 0
Run WQNet= 0
Run RASMapper= 0
UNET Theta= 0
UNET Theta Warmup= 0
UNET ZTol= 0
UNET ZSATol= 0
UNET MxIter= 0
UNET Max Iter WO Improvement= 0
UNET MaxInSteps= 0
UNET DtIC= 0
UNET DtMin= 0
UNET MaxCRTS= 0
UNET WFStab= 0
UNET SFStab= 0
UNET WFX= 1
UNET SFX= 1
UNET Gravity=32.17405
UNET 1D Methodology=Finite Difference
UNET DSS MLevel= 1
UNET Pardiso=0
UNET DZMax Abort= 0
UNET Use Existing IB Tables= 0
UNET Froude Reduction=False
UNET Froude Limit= 0
UNET Froude Power= 0
UNET D1 Cores= 0
UNET WindReference=Eulerian
UNET WindDragFormulation=Hsu (1988)
UNET D2 Coriolis=0
UNET D2 Cores= 0
UNET D2 Theta= 1
UNET D2 Theta Warmup= 1
UNET D2 Z Tol= 0.01
UNET D2 Volume Tol= 0.01
UNET D2 Max Iterations= 20
UNET D2 Equation= 0
UNET D2 RampUpFraction=0.1
UNET D2 TimeSlices= 1
UNET D2 Turbulence Formulation=Non-Conservative (original)
UNET D2 Eddy Viscosity=0.3
UNET D2 Transverse Eddy Viscosity=0.1
UNET D2 Smagorinsky Mixing=0
UNET D2 BCVolumeCheck=0
UNET D2 Cores=0
UNET D2 SolverType=PARDISO (Direct)
UNET D2 Minimum Iterations= 3
UNET D2 Maximum Iterations= 30
UNET D2 Restart Number= 10
UNET D2 Relaxation Coeff=1.3
UNET D2 SOR Precondition Iterations= 10
UNET D2 ILUT Maximum Fill= 8
UNET D2 ILUT Tolerance=1E-08
UNET D2 Convergence Tolerance=0.00001
UNET D1D2 MaxIter= 0
UNET D1D2 ZTol=0.01
UNET D1D2 QTol=0.1
UNET D1D2 MinQTol=1
DSS File=dss
Write IC File= 0
Write IC File at Fixed DateTime=0
Write IC File at Sim End=0
Echo Input=False
Echo Parameters=False
Echo Output=False
Write Detailed= 0
HDF Write Warmup=0
HDF Write Time Slices=0
HDF Flush=0
HDF Compression= 1
HDF Chunk Size= 1
HDF Spatial Parts= 1
HDF Use Max Rows=0
HDF Fixed Rows= 1
Calibration Method= 0
Calibration Iterations= 20
Calibration Max Change=0.05
Calibration Tolerance=0.2
Calibration Maximum=1.5
Calibration Minimum=0.5
Calibration Optimization Method= 1
WQ AD Non Conservative
WQ ULTIMATE=-1
WQ Max Comp Step=1HOUR
WQ Output Interval=15MIN
WQ Output Selected Increments= 0
WQ Output face flow=0
WQ Output face velocity=0
WQ Output face area=0
WQ Output face dispersion=0
WQ Output cell volume=0
WQ Output cell surface area=0
WQ Output cell continuity=0
WQ Output cumulative cell continuity=0
WQ Output face conc=0
WQ Output face dconc_dx=0
WQ Output face courant=0
WQ Output face peclet=0
WQ Output face adv mass=0
WQ Output face disp mass=0
WQ Output cell mass=0
WQ Output cell source sink temp=0
WQ Output nsm pathways=0
WQ Output nsm derived pathways=0
WQ Create Restart=0
WQ Fixed Restart=0
WQ System Summary=0
WQ Write To DSS=0
Sorting and Armoring Iterations= 10
XS Update Threshold= 0.02
Bed Roughness Predictor= 0
Hydraulics Update Threshold= 0.02
Energy Slope Method= 1
Volume Change Method= 1
Sediment Retention Method= 0
Sediment TS Multiplier= 1
Warm Up Method= 0
XS Weighting Method= 0
Number of US Weighted Cross Sections= 1
Number of DS Weighted Cross Sections= 1
Upstream XS Weight=0
Main XS Weight=1
Downstream XS Weight=0
Number of DS XS's Weighted with US Boundary= 1
Upstream Boundary Weight= 1
Weight of XSs Associated with US Boundary= 0
Number of US XS's Weighted with DS Boundary= 1
Downstream Boundary Weight= 0.5
Weight of XSs Associated with DS Boundary= 0.5
Percentile Method= 0
Sediment Output Level= 3
Mass or Volume Output= 0
Output Increment Type= 1
Profile and TS Output Increment= 1
Transport Output Increment 1
XS Output Flag= 0
XS Output Increment= 10
Read HDF5 Sediment Hotstart= 0
Sediment Hotstart Type= 0
Write Gradation File= 0
Read Gradation Hotstart= 0
Write HDF5 File= 1
Write Binary Output= 1
Write DSS Sediment File= 0
DSS Sediment Output Type= 1
SV Curve= 0
Specific Gage Flag= 0
Subcell Erosion Methods= 0
Subcell Deposition Methods= 0
Advection Scheme= 1
Matrix Solver= 0
Implicit Weighting Factor= 1
Maximum Outer Loop Convergence Iterations= 5
Convergence Maximum Absolute= 0.001
Convergence RMSE= 0.0001
Grain Fractions Max Abs Error= 0.001
Max Subgrid Regions= 1
Max Subgrid Length Scale= 3.402823E+38
Initial Layer Thickness= 3.402823E+38
Min Layer Thickness= 3.402823E+38
Max Layer Thickness= 3.402823E+38
Number of Layers= 5

--- SUGARRN.f01 (steady flow) ---

Flow Title=Flow
Program Version=4.00
Number of Profiles=1
Profile Names=F01pct
River Rch & RM=SUGARRN,Main,31253
     374
River Rch & RM=SUGARRN,Main,29090
     562
River Rch & RM=SUGARRN,Main,27466
     680
River Rch & RM=SUGARRN,Main,25771
     779
River Rch & RM=SUGARRN,Main,24080
     998
River Rch & RM=SUGARRN,Main,22002
    1110
River Rch & RM=SUGARRN,Main,19784
    1240
River Rch & RM=SUGARRN,Main,17000
    1430
River Rch & RM=SUGARRN,Main,14001
    1610
River Rch & RM=SUGARRN,Main,11374
    1800
River Rch & RM=SUGARRN,Main,4002
    2000
Boundary for River Rch & Prof#=SUGARRN,Main      ,1
Up Type=0
Dn Type=3
Dn Slope=0.008623

--- SUGARRN.g01 (geometry) ---

Geom Title=Geometry
Program Version=6.31

River Reach=SUGARRN         ,Main
Reach XY= 30
1677985.83131577416719.0070186911678724.79418873417940.005157558
1678649.18127404418660.554070737 1678901.1725511418771.928114105
1679248.26871098419984.0997630081680056.74971098420921.368763008
1681168.01571098421673.0767630081681112.29471098422659.232763008
1680388.44671098423748.4207630081680218.12971098425032.631763008
1679884.32971098425278.1197630081680112.99571098425517.299763008
1680144.53671098426266.3787630081679485.34671098427215.212763008
1679501.11671098428269.7067630081680142.43371098429933.976763008
1679958.44871098430826.0387630081680615.01071098431672.892763008
1680246.51571098432771.0167630081680328.52071098433613.139763008
1679729.78271098434650.2857630081679582.06971098435827.260763008
1678960.20171098436443.8707630081678674.23771098437312.277763008
1677896.77271098437452.1057630081677800.57471098438108.141763008
1677020.48071098438750.5107630081676870.66471098439521.667763008
1677089.34371098440566.1737630081676217.38971098441761.589763008

Type RM Length L Ch R = 1 ,31253   ,167.6,171.5,167.4
BEGIN DESCRIPTION:
Structure 15 XS 4
END DESCRIPTION:
XS GIS Cut Line= 2
1677801.85844158416899.354773482 1678141.9343154416595.571581845
#Sta/Elev= 30
       0 1185.75    20.6 1184.31    28.2 1182.89    40.6 1182.44    56.7 1180.16
    88.6 1178.59    99.6 1177.29   137.1 1177.22   184.9 1174.39   201.9 1172.67
   249.7  1171.7  253.111171.046   258.6 1169.95   264.2 1171.04   276.6 1171.56
   280.4 1172.27   284.1 1174.42   292.4 1180.75   298.2 1183.45   304.4 1187.51
   309.5 1190.07   323.7 1195.72   335.6 1196.43   340.5 1200.65   346.4 1207.08
     357 1214.24   399.9 1236.19   411.5 1240.48   437.5 1247.57     456 1250.07
#Mann= 5, -1 ,  0
       0     0.1       0     240    0.06       0  253.11   0.045       0
   264.2    0.06       0     380     0.1       0
Bank Sta=253.11,264.2
XS Rating Curve= 0 ,0
Exp/Cntr(USF)=0,0
Exp/Cntr=0.3,0.1

Type RM Length L Ch R = 1 ,31081.98,38.3,39.5,39.4
BEGIN DESCRIPTION:
Structure 15 XS 3
END DESCRIPTION:
XS GIS Cut Line= 4
1677829.41399657417037.8046351581677928.21074252 416918.84528799
1678173.52239064416756.8723915641678166.80152357 416584.81819453
#Sta/Elev= 30
       0 1202.59     6.8 1200.65      38 1195.26    84.8 1188.16   127.8 1182.81
   144.8 1177.91   150.5 1176.89   168.9 1176.39   192.9 1176.86     236 1174.65
   274.4 1171.12   298.3 1170.41   322.3 1170.65   325.8 1170.02   331.9 1168.63
   338.1 1170.03     367 1171.23   383.9 1175.06   391.1 1176.08   424.7 1176.62
   468.9 1181.17     497 1182.69     505 1184.95     513 1186.27     525 1192.19
   547.5 1205.28     561 1214.21     581 1225.35   600.5 1234.01   620.8  1247.1
#Mann= 5, -1 ,  0
       0     0.1       0   325.8   0.045       0   338.1     0.1       0
  344.64    0.06       0   568.6     0.1       0
Bank Sta=325.8,338.1
XS Rating Curve= 0 ,0
Exp/Cntr(USF)=0,0
Exp/Cntr=0.3,0.1

Type RM Length L Ch R = 1 ,31042.47,181.1,194.9,185.2
BEGIN DESCRIPTION:
Structure 15 XS 2
END DESCRIPTION:
XS GIS Cut Line= 4
 1677850.9207712417069.3927103951677949.71751715416950.433363227
1678195.02916527  416788.4604668 1678188.3082982416616.406269767
#Sta/Elev= 30
       0 1208.27     4.3 1207.22    12.8  1203.9    29.9 1201.27    47.9 1196.64
    99.9 1187.19   139.6 1181.88   163.5 1176.19   171.9  1174.8   258.2 1171.21
   272.5 1171.98   282.1 1170.75   325.2 1168.79   339.6 1167.38   346.8 1168.78
     378 1171.69   391.6 1174.39     406 1175.67   448.6 1177.93   468.5 1178.44
   484.5 1179.84   524.6 1181.19   544.6 1184.19   552.6 1186.28   564.6 1191.02
   576.6 1194.51   584.6 1197.74   591.3 1201.67   604.6 1210.71   620.8 1220.23
#Mann= 5, -1 ,  0
       0     0.1       0   325.2   0.045       0   346.8     0.1       0
  354.64    0.06       0   498.6     0.1       0
Bank Sta=325.2,346.8
XS Rating Curve= 0 ,0
Exp/Cntr(USF)=0,0
Exp/Cntr=0.3,0.1

Type RM Length L Ch R = 1 ,30847.57,568.1,585.4,570.9
BEGIN DESCRIPTION:
Structure 15 XS 1
END DESCRIPTION:
XS GIS Cut Line= 3
1677874.63037281417127.1053384961678259.74586017416867.007028223
1678419.89613233416858.692749679
#Sta/Elev= 30
       0 1216.55    16.3    1212    46.1  1201.4    54.9 1197.66      79 1189.77
   117.6 1178.55   132.1 1175.25   154.7 1171.95   204.5 1169.59   247.6  1168.6
   282.4 1166.42   291.4 1164.96   299.7 1166.48   328.5 1168.33   340.5  1168.2
   407.2 1173.25   426.3 1175.96   435.1 1178.64   440.5 1179.46     461 1180.02
   463.9 1180.81   473.1 1185.48   489.1 1184.37   497.1 1184.83   529.2 1193.95
     555 1198.89   585.3 1205.81   609.3  1213.3   617.3 1216.39   625.1 1220.33
#Mann= 5, -1 ,  0
       0     0.1       0   282.4   0.045       0   299.7     0.1       0
  484.72    0.06       0  584.72     0.1       0
Bank Sta=282.4,299.7
XS Rating Curve= 0 ,0
Exp/Cntr(USF)=0,0
Exp/Cntr=0.3,0.1

Type RM Length L Ch R = 1 ,30262   ,556,571.3,554.5
XS GIS Cut Line= 6
1678039.90658326417454.3235258461678186.43647392417342.189891845
1678255.79165018417307.3438329251678337.84726034417245.961081669
1678500.15172575417194.2594134211678589.13448742417160.354625583
#Sta/Elev= 30
       0  1249.1    20.9 1240.21    51.9 1231.99    77.7 1223.06     108 1210.22
   122.8 1205.19   132.6 1199.77   162.1 1192.12   172.7 1190.69   216.9 1180.22
   258.1 1165.63   282.6 1161.34   292.6 1161.51  296.671160.393   302.6 1159.05
   307.6  1160.4   332.6 1161.19   400.5 1159.96   425.6 1162.18     438 1168.03
   463.6 1186.09   480.2    1194   488.6 1199.42   495.3 1201.28   511.1  1202.2
   522.4 1210.98   551.9 1227.69   579.8 1237.12   616.3 1258.59   630.3 1261.55
#Mann= 7, -1 ,  0
       0     0.1       0  204.61    0.05       0  292.22     0.1       0
  296.67   0.045       0   307.6     0.1       0   414.7    0.06       0
  514.91     0.1       0
Bank Sta=296.67,307.6
XS Rating Curve= 0 ,0
Exp/Cntr(USF)=0,0
Exp/Cntr=0.3,0.1

Type RM Length L Ch R = 1 ,29691   ,291.6,307.4,297.3
BEGIN DESCRIPTION:
Structure 14 XS 4
END DESCRIPTION:
XS GIS Cut Line= 6
1678289.99842969417802.2503366711678446.07981045417707.869619915
 1678605.5135467417635.6988325071678676.49207928417610.135891507
1678756.63233895417571.516874248 1678840.5524467417526.311256001
#Sta/Elev= 30
       0 1239.16    20.2  1230.5    37.6 1221.16    69.5 1214.25      84 1205.12
   116.1 1193.02   129.3 1187.22   180.5 1171.16   211.1 1163.52   233.2 1158.94
   273.9 1155.01     299 1154.75   310.3 1153.76   316.3 1153.27   323.61153.764
   390.1 1154.44   398.5 1154.95   408.8 1157.06   419.7  1162.8   432.5 1172.55
   436.9 1173.52   450.2 1173.62   454.7 1174.67   463.5 1183.91   475.7 1192.16
   499.1 1199.26   517.7 1206.17     565 1230.01     594 1241.74   617.2 1254.99
#Mann= 5, -1 ,  0
       0     0.1       0   310.3   0.045       0   323.6     0.1       0
  432.89    0.06       0  541.85     0.1       0
Bank Sta=310.3,323.6
XS Rating Curve= 0 ,0
Exp/Cntr(USF)=0,0
Exp/Cntr=0.3,0.1

Type RM Length L Ch R = 1 ,29383   ,40.9,40.4,44.8
BEGIN DESCRIPTION:
Structure 14 XS 3
END DESCRIPTION:
XS GIS Cut Line= 6
1678400.80361805417928.8196523841678589.73465907 417853.39658858
1678665.15772287417876.5462418261678703.98939928417880.280056866
1678818.99090251417904.9232361291678950.42119191417698.069882924
#Sta/Elev= 30
       0 1226.27    42.3 1206.18    59.6 1199.44    72.5 1193.76    85.4 1189.51
    95.1  1184.6   132.8 1174.34   165.9 1166.59   203.4 1160.44   243.6  1155.7
   264.5 1152.64   297.4 1151.46   305.4 1150.41  311.561151.435   325.6 1151.76
   354.2    1151   423.7  1150.8   458.4 1151.83   478.3    1154   491.5 1153.62
   495.1 1154.02   506.7 1157.92   524.7  1163.2   538.6 1165.92   548.4 1168.98
   561.8 1172.22   627.5 1192.06   666.1 1202.45   676.4 1206.74     684 1210.51
#Mann= 7, -1 ,  0
       0     0.1       0      10    0.05       0     190     0.1       0
   297.4   0.045       0  311.56     0.1       0  391.34    0.05       0
  538.95     0.1       0
Bank Sta=297.4,311.56
XS Rating Curve= 0 ,0
Exp/Cntr(USF)=0,0
Exp/Cntr=0.3,0.1

Type RM Length L Ch R = 1 ,29343.08,239.4,253,237
BEGIN DESCRIPTION:
Structure 14 XS 2
END DESCRIPTION:
XS GIS Cut Line= 6
1678414.24535219 417951.969305631678571.06558387417888.494449954
1678688.30737612417913.8843922241678739.08726066417921.352022304
1678835.41968868417940.7678605111678975.81113418417707.777802028
#Sta/Elev= 30
       0 1226.88    40.9 1206.27    75.4 1191.88      87 1188.94      97    1185
   140.1 1174.56   169.4 1166.47   182.5 1164.03   202.9 1159.38     256 1152.76
   276.6  1151.3     293 1151.14   297.1 1150.68   305.1 1149.46   317.3 1150.74
   386.6 1150.06   410.8 1150.43   448.3 1151.37   462.5 1152.55   490.5 1153.75
   504.5 1153.22   513.8 1154.28   532.5 1158.64   540.9 1159.73   550.2 1162.98
   560.5  1165.6   585.2 1170.43   649.3 1190.76   691.3 1202.26   710.9 1210.58
#Mann= 8, -1 ,  0
       0     0.1       0      70    0.05       0  179.18     0.1       0
   297.1   0.045       0   317.3     0.1       0  380.49    0.05       0
  508.83    0.06       0  578.83     0.1       0
Bank Sta=297.1,317.3
XS Rating Curve= 0 ,0
Exp/Cntr(USF)=0,0
Exp/Cntr=0.3,0.1

Type RM Length L Ch R = 1 ,29090   ,502.8,503,497.3
BEGIN DESCRIPTION:
Structure 14 XS 1
END DESCRIPTION:
XS GIS Cut Line= 6
1678399.27069393418009.4989246731678494.79314068418020.597327679
1678579.14205334418046.8449785861678739.09711401 418126.77362451
 1678816.6697935418154.8260618451678999.65663226418209.699967846
#Sta/Elev= 30
       0 1238.42    12.9 1235.59    41.1 1232.68    49.2 1231.07    61.3 1227.75
    77.4 1222.61    97.5 1214.38   114.3 1208.79   143.6 1200.75   156.2 1195.79
     173 1191.36   185.6 1184.99   190.1 1183.39   235.5  1170.9   258.2 1166.76
   266.4 1164.57   275.4 1160.84   289.2  1152.8   293.6 1150.77   302.5 1148.46
   311.5 1147.71   320.2 1146.95  323.921147.739   329.1 1148.49   415.4 1148.03
   456.4 1148.43   517.1 1150.11   536.3 1152.04   624.9 1166.62   636.9 1169.07
#Mann= 5, -1 ,  0
       0     0.1       0   311.5   0.045       0  323.92     0.1       0
  359.97    0.05       0  609.15    0.06       0
Bank Sta=311.5,323.92
XS Rating Curve= 0 ,0
Exp/Cntr(USF)=0,0
Exp/Cntr=0.3,0.1

Type RM Length L Ch R = 1 ,28587   ,576.5,584.6,564.1
XS GIS Cut Line= 6
 1678335.1195755418571.5588241671678428.81787892418574.672663093
1678516.26980376418577.5778409991678591.22831526418580.068321586
1678691.17299725 418583.389837251679027.59154793418569.959811973
#Sta/Elev= 30
       0 1205.79      73 1196.53   133.1 1184.84   185.1 1179.18   197.1 1177.23
   241.1 1164.84   285.2 1156.63   293.2  1152.9   297.2 1150.24   301.2 1146.61
   306.4 1143.62   317.2 1142.04   322.9 1143.63   329.2 1144.53   373.2 1143.17
   453.3  1143.4   481.3 1145.24   493.3 1147.66   517.3 1155.29   533.3 1159.02
   557.4 1162.89   585.4 1169.43   609.4 1172.82   613.4 1174.19   621.4  1178.9
   629.4 1180.19   641.4 1180.26   645.4 1181.03   661.4 1193.26   692.9 1201.83
#Mann= 6, -1 ,  0
       0     0.1       0   306.4   0.045       0   322.9     0.1       0
  446.25    0.05       0  536.25     0.1       0  636.25    0.06       0
Bank Sta=306.4,322.9
XS Rating Curve= 0 ,0
Exp/Cntr(USF)=0,0
Exp/Cntr=0.3,0.1

Type RM Length L Ch R = 1 ,28003   ,533.8,536.2,535.3
BEGIN DESCRIPTION:
Structure 13 XS 4
END DESCRIPTION:
XS GIS Cut Line= 6
1678635.21707243419005.436893418  1678719.045973418948.391403839
1678803.65374343418915.1460635071678877.45838584418896.515851423
1679120.95428993418798.1682790821679210.25463626418768.763482258
#Sta/Elev= 30
       0 1149.67     5.9 1148.05     9.9 1147.86   115.4 1148.02   198.1 1146.32
   217.5 1144.46   238.2 1139.61     297 1139.54   305.5 1138.95   310.7 1137.16
   314.1 1136.36   322.7 1137.21   339.8 1142.61   349.5 1147.94   378.5 1161.14
   391.5 1170.46   395.8 1172.03   400.1  1172.5   417.5 1172.81   421.8 1174.87
   426.1 1179.19   430.5 1182.49   434.8 1184.41   489.3 1202.11   517.1 1210.25
   555.4 1226.94   572.9 1232.13   601.8 1242.88   614.1  1248.4   625.1 1254.79
#Mann= 5, -1 ,  0
       0    0.05       0   262.3    0.06       0   310.7   0.045       0
   322.7    0.06       0  368.42     0.1       0
Bank Sta=310.7,322.7
XS Rating Curve= 0 ,0
Exp/Cntr(USF)=0,0
Exp/Cntr=0.3,0.1

Type RM Length L Ch R = 1 ,27466   ,40.9,41.9,42.4
BEGIN DESCRIPTION:
Structure 13 XS 3
END DESCRIPTION:
XS GIS Cut Line= 3
1678724.73545201419405.2418619731679127.31139457419357.096647468
1679455.10859971419267.976782321
#Sta/Elev= 30
       0  1145.4    19.5 1145.19    39.7 1143.69   124.3 1139.53   148.4 1139.85
   160.5 1137.52   176.6 1138.51   301.5 1135.66   309.6 1136.69   320.3 1136.76
   341.8 1135.21   409.8 1133.52   418.7 1132.66   422.9 1132.91  424.711133.583
   435.3 1137.87   443.6 1139.85   451.9 1140.64   472.6 1141.22   494.6 1143.78
   510.8 1144.74   543.1 1149.35   559.5 1150.17   595.6 1149.17   613.5  1149.5
   667.4 1155.65   688.2 1156.44   729.2 1159.15   737.9 1158.42   745.1 1159.94
#Mann= 6, -1 ,  0
       0    0.05       0     350    0.08       0   409.8   0.045       0
  424.71    0.08       0  445.44    0.05       0  555.44     0.1       0
Bank Sta=409.8,424.71
XS Rating Curve= 0 ,0
Exp/Cntr(USF)=0,0
Exp/Cntr=0.3,0.1

Type RM Length L Ch R = 1 ,27424   ,9.2,6.7,7.3
BEGIN DESCRIPTION:
Structure 13 XS 2
END DESCRIPTION:
XS GIS Cut Line= 4
 1678743.1740448419446.2165126151679137.55505723419396.022565578
 1679199.0170332419379.6327053211679459.20606478419304.853967899
#Sta/Elev= 30
       0 1149.31    21.1 1148.71   113.9 1142.18   214.7 1137.12   307.4  1135.4
   342.2 1136.25     409 1134.11   420.9 1132.12   425.4 1132.46   430.1 1134.08
   438.5 1138.69   441.6 1139.43     454 1140.31   458.2 1141.51   466.5 1145.69
   474.8 1148.47   491.4 1150.79   574.7 1154.75   599.7 1158.21   620.5    1164
   639.1 1162.67   649.6  1163.2   662.1 1166.22   678.7 1171.27   691.2 1172.44
   707.9 1172.87   716.2 1172.33   720.4 1171.69   728.7 1168.24   731.9 1167.63
#Mann= 6, -1 ,  0
       0    0.05       0     330    0.06       0     350    0.08       0
     409   0.045       0   430.1    0.05       0  531.17     0.1       0
Bank Sta=409,430.1
XS Rating Curve= 0 ,0
Exp/Cntr(USF)=0,0
Exp/Cntr=0.3,0.1

Type RM Length L Ch R = 1 ,27418   ,64.8,71,74.8
BEGIN DESCRIPTION:
Structure 12 XS 4 AND Structure 13 XS 1
END DESCRIPTION:
XS GIS Cut Line= 3
1678752.39334119419459.533274074 1679144.7256211419399.095664376
1679466.37662864419345.828618541
#Sta/Elev= 30
       0    1152      24 1150.66    68.5 1146.14   209.3 1137.04   299.2 1135.15
     318 1135.12   343.7 1136.23   384.2 1134.29   402.1 1134.23   409.1 1133.28
   416.6 1132.25  422.731133.284   432.8 1138.89     449 1140.42   461.2 1146.56
   469.3 1149.12   478.7 1150.82   497.7 1153.18   537.8 1154.16   542.3 1156.14
   546.4 1157.02     595 1165.81   619.3 1167.12   627.4 1168.51   639.6 1172.27
   647.7    1174     672 1176.46   684.7 1176.19   699.2 1179.43     723 1183.49
#Mann= 7, -1 ,  0
       0    0.05       0     320    0.06       0     380    0.08       0
   409.1   0.045       0  422.73    0.08       0  426.96    0.05       0
  526.96     0.1       0
Bank Sta=409.1,422.73
XS Rating Curve= 0 ,0
Exp/Cntr(USF)=0,0
Exp/Cntr=0.3,0.1

Type RM Length L Ch R = 1 ,27347   ,78.3,82.4,88.4
BEGIN DESCRIPTION:
Structure 12 XS 3
END DESCRIPTION:
XS GIS Cut Line= 5
1678786.19742798419587.5790573321679111.94590058419406.266228239
1679158.04238255419454.4114427441679197.99266693419480.020599395
1679477.64465757419447.240878881
#Sta/Elev= 30
       0  1171.1    30.1 1167.01    89.2 1154.99   139.5 1147.09   180.1 1138.93
     199 1136.65   224.2 1135.38   312.4 1134.71     336 1134.84   353.6 1136.28
   368.1 1135.38   436.7 1135.55   450.8 1133.42   458.2 1131.92   465.6 1133.47
     483 1139.61   501.1 1140.55   505.2  1142.3   521.3 1151.96   525.3  1153.2
   549.5 1155.31   578.5 1160.81   609.9 1165.36   638.1 1172.15   658.2 1175.18
   706.5 1186.22   726.7 1188.34   750.8 1188.97   754.9 1189.95   768.5 1196.29
#Mann= 7, -1 ,  0
       0    0.05       0     330    0.06       0  449.46    0.05       0
   450.8   0.045       0   465.6    0.05       0  656.92    0.07       0
  756.92     0.1       0
Bank Sta=450.8,465.6
XS Rating Curve= 0 ,0
Exp/Cntr(USF)=0,0
Exp/Cntr=0.3,0.1

Type RM Length L Ch R = 1 ,27264   ,195.2,184.9,173.1
BEGIN DESCRIPTION:
Structure 12 XS 2
END DESCRIPTION:
XS GIS Cut Line= 6
1678804.63602076419617.2856790471679104.77533672419467.728204203
1679128.33576084419491.2886283221679154.96928376419519.970883772
 1679199.0170332419574.2622958731679474.57155877419530.214546432
#Sta/Elev= 30
       0  1173.3      36 1167.18      62 1161.81     129 1150.94   142.4 1147.34
   173.7 1137.16   187.1 1134.99   217.9 1133.39   362.7 1133.28   411.9 1133.89
   426.1 1133.46   431.8 1132.29     435 1131.14   441.4 1130.36   447.7  1130.6
  454.791132.366   466.8  1137.4   478.8 1140.61   515.3 1144.16   519.3 1145.17
   527.4 1149.89   531.5 1151.17   580.1 1160.86   600.3 1166.06   616.4 1167.69
   636.8 1173.35   689.7 1185.02   705.7 1186.56     718 1190.71   756.8 1200.32
#Mann= 9, -1 ,  0
       0    0.05       0     300    0.06       0  388.66    0.05       0
   427.8    0.06       0   431.8   0.045       0  454.79    0.06       0
  547.71    0.05       0  647.71     0.1       0  747.71    0.05       0
Bank Sta=431.8,454.79
XS Rating Curve= 0 ,0
Exp/Cntr(USF)=0,0
Exp/Cntr=0.3,0.1

Type RM Length L Ch R = 1 ,27080   ,330.6,331.2,325.1
BEGIN DESCRIPTION:
Structure 12 XS 1
END DESCRIPTION:
XS GIS Cut Line= 2
 1678909.1213799419788.3548454791679485.83958769419659.284695956
#Sta/Elev= 30
       0 1178.79    76.8 1157.34   130.1 1145.25   162.9 1134.51   171.1 1132.77
   220.3 1128.66   232.6 1129.57   261.3 1129.25   302.3 1130.52   307.1 1130.03
   317.2 1127.95   318.7    1128  321.111130.112   322.8 1131.56   326.9 1136.86
     331 1138.66   350.7 1139.39   359.7 1144.99   367.4 1147.88   376.1 1148.89
   400.9 1155.44   457.9 1167.64   470.3 1171.87   503.1 1172.99   515.4 1179.31
   519.5 1180.67   531.8 1183.69     540 1184.67   552.3 1189.83     591 1201.61
#Mann= 6, -1 ,  0
       0    0.05       0     270     0.1       0   307.1   0.045       0
  321.11     0.1       0     420    0.05       0     570     0.1       0
Bank Sta=307.1,321.11
XS Rating Curve= 0 ,0
Exp/Cntr(USF)=0,0
Exp/Cntr=0.3,0.1

Type RM Length L Ch R = 1 ,26748   ,195.9,191.7,179.3
BEGIN DESCRIPTION:
Structure 11 XS 4
END DESCRIPTION:
XS GIS Cut Line= 2
1679053.55702342420140.7368410041679581.10565044419856.987385305
#Sta/Elev= 30
       0 1183.85    25.6  1177.6      68 1170.88   111.9 1158.84     132 1155.08
   146.8 1150.68   157.3 1144.29   160.9 1143.21   199.9  1139.9   202.9 1139.02
   214.7 1132.47   225.5 1128.66   247.2 1127.18   266.3 1126.73   279.1 1125.26
   285.6 1124.18     289 1124.22  293.131125.304   303.3 1129.85   315.1 1130.57
   325.4 1130.11   329.9 1130.94   334.5  1133.2   348.1 1142.99   365.3 1149.12
   380.1 1150.57   486.4 1173.76   507.1 1180.09   548.4 1195.12     599 1209.57
#Mann= 8, -1 ,  0
       0     0.1       0      20    0.05       0     110    0.06       0
     130    0.05       0     240    0.06       0   279.1   0.045       0
  293.13    0.06       0     360     0.1       0
Bank Sta=279.1,293.13
XS Rating Curve= 0 ,0
Exp/Cntr(USF)=0,0
Exp/Cntr=0.3,0.1

Type RM Length L Ch R = 1 ,26557   ,53.2,54,54.7
BEGIN DESCRIPTION:
Structure 11 XS 3
END DESCRIPTION:
XS GIS Cut Line= 6
1679330.37742218420510.9523034611679431.54939907420298.491151982
1679404.99175514420144.2038872171679377.16946149420094.882548481
1679348.08251813420058.2077068561679617.45290662419879.892097579
#Sta/Elev= 30
       0 1163.14    41.3 1158.64   100.1 1147.47   135.6 1142.59     171 1133.63
   193.2 1129.34     202 1126.16   215.3 1125.41   225.2 1126.53   235.3 1126.14
   285.4 1127.33   366.8 1125.32   375.51124.038   379.4 1122.56   387.7 1124.02
   407.3 1125.36   479.7 1125.31   495.7 1125.95   508.4 1128.65   528.6 1129.65
   540.2    1136   554.6 1138.47   567.6 1147.21   589.2 1150.64   690.3 1172.29
   716.1 1180.34   762.4 1196.86   797.9 1207.14   810.3 1211.89   818.7 1216.42
#Mann= 5, -1 ,  0
       0    0.05       0  255.32    0.06       0   375.5   0.045       0
   387.7    0.06       0  615.64     0.1       0
#XS Ineff= 2 , 0
          281.81 1146.55
Permanent Ineff=
       F       F
Bank Sta=375.5,387.7
XS Rating Curve= 0 ,0
Exp/Cntr(USF)=0,0
Exp/Cntr=0.3,0.1

Type RM Length L Ch R = 1 ,26503   ,254.6,257.4,262.8
BEGIN DESCRIPTION:
Structure 11 XS 2
END DESCRIPTION:
XS GIS Cut Line= 6
1679377.16946149420528.6573994171679494.78188463420327.578095339
1679474.54748925420284.5800051591679455.57774359420154.321084907
1679406.25640485420065.7956051241679645.27520026419903.920442092
#Sta/Elev= 30
       0 1159.97    83.6 1150.27   139.2 1142.11   162.3 1140.27   177.7 1136.03
   195.2 1126.15   212.8 1126.55   232.9 1124.42   258.4 1124.85   267.3 1123.47
   276.3 1125.45   296.6 1123.91   373.8 1124.46  385.551122.105     398 1122.04
     406 1121.41   428.4 1125.09   470.3 1129.09   484.2 1131.45   514.6 1133.24
   531.3    1142   545.4 1147.15   560.4 1149.47   618.3 1163.94   652.3  1170.5
   676.3 1176.23   695.5 1181.65   743.9 1198.52   784.8 1209.72   803.3 1217.51
#Mann= 7, -1 ,  0
       0    0.05       0     170    0.06       0  280.47     0.1       0
  377.73    0.06       0  385.55   0.045       0     398    0.06       0
  584.64     0.1       0
Bank Sta=385.55,398
XS Rating Curve= 0 ,0
Exp/Cntr(USF)=0,0
Exp/Cntr=0.3,0.1

Type RM Length L Ch R = 1 ,26245   ,243.7,245.2,246.1
BEGIN DESCRIPTION:
Structure 11 XS 1
END DESCRIPTION:
XS GIS Cut Line= 2
1679478.61639762420568.867474941 1679821.4891634420109.722068244
#Sta/Elev= 30
       0 1148.48    42.6 1145.45   109.9 1142.74   145.2 1140.67   150.2 1139.92
   155.2  1136.6   158.5  1133.4   161.4 1131.59   164.2 1131.04   175.1 1130.46
   178.5 1129.72   189.7 1123.57   195.1 1122.29   215.1 1121.36     255 1122.11
     260 1121.44   264.2 1119.81   267.1 1119.58     270    1120  273.351121.465
   284.2 1128.07     290    1131   309.9 1137.65   379.8 1154.42     437 1165.39
   447.2 1166.71   474.7 1174.42   514.6 1187.95   554.6 1199.12     573 1205.36
#Mann= 5, -1 ,  0
       0    0.05       0     110    0.06       0     230     0.1       0
     260   0.045       0  273.35     0.1       0
Bank Sta=260,273.35
XS Rating Curve= 0 ,0
Exp/Cntr(USF)=0,0
Exp/Cntr=0.3,0.1

Type RM Length L Ch R = 1 ,26000   ,174.3,178.9,183.3
BEGIN DESCRIPTION:
Structure 10 XS 4
END DESCRIPTION:
XS GIS Cut Line= 3
1679596.99407385420562.2734707251679820.07828291420501.949679501
1680007.87876502420282.280024668
#Sta/Elev= 30
       0 1141.58    36.4 1140.71    61.2 1140.82    98.6 1138.68     111 1136.63
   129.2 1131.53   144.2 1130.99   160.5 1129.41   181.4  1128.1   199.7 1124.85
   237.3 1124.38   243.5 1122.78   249.6 1120.42   255.8 1118.91   260.5  1118.6
   269.8 1118.97  273.241118.586   280.4    1117   291.7 1118.57   297.4 1119.49
   301.4 1120.95   322.9 1136.27   332.9 1141.78   343.5 1145.15   354.3 1146.78
   379.7 1151.79     408 1156.09     454 1161.61   469.8 1164.12   520.1 1169.72
#Mann= 5, -1 ,  0
       0    0.06       0     170    0.05       0   261.1     0.1       0
  273.24   0.045       0   291.7     0.1       0
Bank Sta=273.24,291.7
XS Rating Curve= 0 ,0
Exp/Cntr(USF)=0,0
Exp/Cntr=0.3,0.1

Type RM Length L Ch R = 1 ,25821   ,50,50,50.2
BEGIN DESCRIPTION:
Structure 10 XS 3
END DESCRIPTION:
XS GIS Cut Line= 6
1679591.92149661420597.0896877911679806.25417019420602.134059088
1679892.75621043420610.1013522681679932.59267634420611.239537008
1679980.39643542420599.8576896081680214.41004125420501.925557041
#Sta/Elev= 30
       0 1143.08    12.2 1143.45    60.2 1141.91    84.2 1140.16   120.2 1136.64
   144.2 1133.72   176.2 1125.62   196.2 1125.66   224.3 1122.83   308.6 1117.76
   341.1 1117.46   357.1 1118.12   362.9 1117.12   366.2 1116.03   369.4 1115.66
  375.241117.098   377.6 1117.83   381.7 1118.19   394.3 1118.59   411.5 1118.36
   420.1 1118.83   428.8 1119.95   438.7 1122.87   454.6 1128.83   476.2 1135.47
     511 1143.78   550.1 1150.71   597.5 1156.82   619.7 1158.32   643.9 1162.57
#Mann= 5, -1 ,  0
       0    0.06       0  264.39    0.05       0   362.9   0.045       0
  375.24     0.1       0  582.47    0.05       0
Bank Sta=362.9,375.24
XS Rating Curve= 0 ,0
Exp/Cntr(USF)=0,0
Exp/Cntr=0.3,0.1

Type RM Length L Ch R = 1 ,25771   ,274.2,270.7,264.7
BEGIN DESCRIPTION:
Structure 10 XS 2
END DESCRIPTION:
XS GIS Cut Line= 6
1679611.43653303420643.7311396731679825.76920661 420648.77551097
1679912.27124685 420656.742804151679952.10771276 420657.88098889
1679999.91147184 420646.499141491680233.92507767420548.567008923
#Sta/Elev= 30
       0 1143.84    80.7 1134.41    87.5 1133.22    96.7 1130.65   106.4 1128.74
   128.7 1125.86   144.7 1122.34   160.7 1123.13   172.7 1122.95   185.2 1121.96
   204.7 1119.19   240.8  1117.5   271.5  1117.2   345.2  1117.8   349.3 1117.49
   352.2 1116.71   357.6 1115.16   361.7 1114.85   365.8  1115.1  372.48 1116.74
   382.2 1120.64   386.3 1121.84   425.7 1127.51   444.9 1130.87   474.9 1137.02
   520.2 1147.87   531.7 1150.04   581.1 1158.23   611.5 1162.17   643.9 1167.02
#Mann= 6, -1 ,  0
       0    0.06       0  244.39    0.05       0  351.11     0.1       0
   352.2   0.045       0  372.48     0.1       0  562.47    0.05       0
Bank Sta=352.2,372.48
XS Rating Curve= 0 ,0
Exp/Cntr(USF)=0,0
Exp/Cntr=0.3,0.1

Type RM Length L Ch R = 1 ,25500   ,499.7,502.2,502.4
BEGIN DESCRIPTION:
Structure 10 XS 1
END DESCRIPTION:
XS GIS Cut Line= 6
1679820.57034476 421115.24369742 1680007.7346686420939.945163503
1680082.96023992420873.6113066671680140.32790734 420815.93228817
1680213.37992659420751.0534809231680295.79413185420687.122178346
#Sta/Elev= 30
       0 1181.97    58.2 1178.97      80 1176.73    97.6 1173.34     121 1166.35
   173.7 1157.18     194 1150.59   202.9 1148.49   208.8 1144.31   214.6 1137.68
   220.5 1134.29   249.7 1135.94   259.1 1134.25     262 1133.18   267.6 1129.58
   279.7 1119.81   287.5 1116.11     296 1113.74   304.9 1111.17   310.3 1111.74
  315.411113.738   320.9 1114.52   341.3  1113.6   431.6 1115.64   465.8 1124.91
   485.9 1132.04   496.6 1135.02   527.5 1141.43   579.7  1154.4   640.1 1165.92
#Mann= 6, -1 ,  0
       0    0.05       0  181.29    0.06       0     296   0.045       0
  315.41    0.06       0  316.44    0.05       0  458.08     0.1       0
Bank Sta=296,315.41
XS Rating Curve= 0 ,0
Exp/Cntr(USF)=0,0
Exp/Cntr=0.3,0.1

Type RM Length L Ch R = 1 ,24998   ,499.7,499.4,495.7
XS GIS Cut Line= 6
1680239.37987459421418.5344294161680355.14473492421275.869032338
1680407.73583709421221.0810841771680487.95450868421161.350232512
1680530.03414892421096.4943910841680609.75183725420925.751294255
#Sta/Elev= 30
       0 1169.79    28.1 1168.87    53.2 1164.55    79.1 1162.48   135.3 1154.03
   188.4  1139.2   193.9 1136.05   203.8 1127.27   208.2 1125.11   229.2 1125.63
   243.4 1124.73   251.8 1122.33   260.6 1116.36   275.1 1109.58  296.131106.258
   303.2 1105.18     320 1106.29     330 1106.83   339.9 1108.95   404.1 1108.42
   432.2 1110.77     437 1112.28   450.8 1121.41     469 1129.82     486 1136.35
   530.5  1145.8   556.7 1153.14   578.6 1155.98     618 1167.55   625.5 1168.57
#Mann= 6, -1 ,  0
       0    0.06       0      20    0.05       0  193.74    0.06       0
  296.13   0.045       0     320    0.06       0  339.68     0.1       0
Bank Sta=296.13,320
XS Rating Curve= 0 ,0
Exp/Cntr(USF)=0,0
Exp/Cntr=0.3,0.1

Type RM Length L Ch R = 1 ,24499   ,418.9,418.9,418.9
BEGIN DESCRIPTION:
Structure 9 XS 4
END DESCRIPTION:
XS GIS Cut Line= 6
1680596.50350417421690.6562605051680662.10311051421623.643927336
1680724.53671268421562.3379475921680778.25281259421509.997173011
1680966.26129484421326.8059383331681033.40682983421261.379560009
#Sta/Elev= 30
       0 1162.83    36.6 1156.01    58.9 1150.23    85.2 1141.93   132.5 1125.27
   152.7 1117.43   166.7 1113.26   190.7 1110.64   219.8 1110.98   246.9 1108.22
   264.1 1107.46   275.6 1105.65   289.7 1104.96   295.4 1104.07   303.6 1102.24
   309.1 1101.74   314.7 1102.56  318.631104.155   326.5  1106.7   344.3 1116.28
   353.8 1119.95   385.9 1129.84   413.1 1139.51   470.4 1156.65   499.1 1163.45
   527.8 1167.86     545  1172.5   558.5 1176.95   583.9 1186.78   612.5 1196.42
#Mann= 6, -1 ,  0
       0    0.06       0      40    0.05       0  181.28    0.06       0
  211.28    0.05       0   295.4   0.045       0  318.63     0.1       0
Bank Sta=295.4,318.63
XS Rating Curve= 0 ,0
Exp/Cntr(USF)=0,0
Exp/Cntr=0.3,0.1

Type RM Length L Ch R = 1 ,24080   ,64.9,64.9,64.9
BEGIN DESCRIPTION:
Structure 9 XS 3
END DESCRIPTION:
XS GIS Cut Line= 6
1680756.00611819421777.8719026361680929.82207775421580.480321441
1681117.84314178421658.5261058551681184.90459058421677.472159449
1681314.91514947421735.5865796121681459.19284005421859.495842196
#Sta/Elev= 30
       0 1145.16    60.7 1131.12    76.4    1126      91 1119.32   108.7 1116.08
     119 1111.13   122.9 1110.27   193.6 1107.63   230.6 1108.69   246.9 1107.33
     263 1103.93   308.8 1103.66     323 1102.05   336.2 1102.93   412.7 1101.66
     430 1103.05   489.1 1101.46   498.6 1102.23   509.9  1098.9     515 1097.88
   531.2  1098.9   546.9 1105.63   557.9 1107.44     686  1108.5   741.7 1110.51
   766.2 1109.36   772.4 1110.72   796.9 1120.39   833.8 1127.69     869 1138.28
#Mann= 9, -1 ,  0
       0    0.05       0     130    0.06       0  273.01    0.07       0
  496.59    0.06       0   509.9   0.045       0   531.2    0.06       0
  596.22    0.08       0  708.83     0.1       0  728.83    0.07       0
Bank Sta=509.9,531.2
XS Rating Curve= 0 ,0
Exp/Cntr(USF)=0,0
Exp/Cntr=0.3,0.1

Type RM Length L Ch R = 1 ,24015   ,518.1,515.1,510.1
BEGIN DESCRIPTION:
Structure 9 XS 2
END DESCRIPTION:
XS GIS Cut Line= 4
1680782.51494317421796.2622633451680906.13695569421651.113361719
1681290.20566114421781.6348295041681433.45898546421919.885219813
#Sta/Elev= 30
       0  1145.4      35 1137.28      58 1128.87    76.5 1125.71   105.9 1114.07
   120.5 1109.32   187.5 1106.48   239.2 1105.81     273 1103.88   293.9  1104.4
   331.8 1102.34   406.4 1101.88     442 1102.69   446.2 1102.35  453.131099.074
   454.7 1098.03   463.1 1096.87   470.8 1099.12   477.1 1101.38   518.1 1104.81
   530.7 1108.88   574.9 1108.77   594.1 1109.76   610.1 1112.67   632.3  1122.2
   653.5 1128.46   698.4 1132.92   737.9 1139.32     779 1142.62   795.4 1147.17
#Mann= 11, -1 ,  0
       0    0.05       0      90    0.06       0  230.66    0.07       0
  240.66    0.06       0  330.66    0.05       0  440.66    0.06       0
  453.13   0.045       0   470.8    0.06       0  540.66    0.08       0
  550.66    0.07       0  795.38    0.05       0
Bank Sta=453.13,470.8
XS Rating Curve= 0 ,0
Exp/Cntr(USF)=0,0
Exp/Cntr=0.3,0.1

Type RM Length L Ch R = 1 ,23500   ,491.8,499.9,504.8
BEGIN DESCRIPTION:
Structure 9 XS 1
END DESCRIPTION:
XS GIS Cut Line= 6
1680819.81736201422246.8424840871680912.08128509422227.436026841
1681173.44657601422203.1030702591681247.93330367422185.522724837
1681334.30616242422156.6628744161681425.22986509422122.898506254
#Sta/Elev= 30
       0 1196.95    28.9 1181.49    45.3 1174.79    53.4  1172.4    90.2 1166.41
   122.4 1159.05   138.5 1153.69   226.9 1104.87   251.5 1099.75   287.1 1098.15
   291.2 1097.66   295.2 1096.04   303.2    1094   311.3 1094.45  315.051096.053
   319.3 1097.58   323.3 1097.64   400.6 1097.04   425.3 1100.98   437.7 1101.42
   446.2 1100.74   450.4 1103.14   458.8 1111.58   488.3 1131.56   492.6 1134.19
   505.2 1139.27   547.6 1152.42   573.2 1159.13   594.3 1163.62   621.4 1167.55
#Mann= 5, -1 ,  0
       0     0.1       0   295.2   0.045       0  315.05     0.1       0
  426.79    0.06       0  523.32     0.1       0
Bank Sta=295.2,315.05
XS Rating Curve= 0 ,0
Exp/Cntr(USF)=0,0
Exp/Cntr=0.3,0.1

Type RM Length L Ch R = 1 ,23000   ,492.8,496.4,498.1
XS GIS Cut Line= 6
1680828.45743659422532.0784621691680918.12425201422567.131213591
1681000.55978267422602.7420347481681067.55669592422638.288879678
1681284.77443734422785.7751332521681367.24015167422831.167102844
#Sta/Elev= 30
       0 1174.77     8.2 1171.23    46.4 1161.09    80.4 1147.38    98.4 1137.36
     108 1130.47   120.2  1126.4   129.3 1119.85   146.4  1109.9   163.8 1102.05
   172.5 1099.46   189.9 1096.52   221.8 1093.87   266.8 1092.49   295.7 1093.77
   301.5 1091.58   310.5 1090.08  320.941091.585   329.7 1098.26   334.5 1099.41
   348.9 1100.39   359.2 1099.22   363.3 1102.08     383 1124.48   415.6 1137.88
   523.7 1166.46     542 1169.91   578.5 1173.19   592.2 1178.41   618.6 1192.31
#Mann= 5, -1 ,  0
       0     0.1       0  226.07    0.06       0   301.5   0.045       0
  320.94    0.06       0  466.97     0.1       0
Bank Sta=301.5,320.94
XS Rating Curve= 0 ,0
Exp/Cntr(USF)=0,0
Exp/Cntr=0.3,0.1

Type RM Length L Ch R = 1 ,22504   ,503.6,501.9,498
XS GIS Cut Line= 6
 1680702.1502745422807.0582271671680759.88277058422887.304129675
 1680800.2957475422966.3991158461680837.42461026423032.460991591
1680895.98092359423113.5805800111681052.22044051423316.689753845
#Sta/Elev= 30
       0 1172.75    37.6 1169.63    58.2 1164.72    68.4 1164.18   104.7 1153.08
   136.2 1141.85   187.7 1118.12   195.5 1113.56   212.6 1100.45   230.2 1090.96
   236.1 1088.82   244.9 1088.13   299.8  1089.5   305.6  1087.7   312.9  1085.2
   317.8 1085.66  322.251087.744   328.5 1091.45   336.4 1092.85   383.4 1094.83
   403.1 1099.28   428.5  1099.6   442.7 1111.22   454.1 1117.62   468.7 1119.32
   513.6 1138.76     526 1142.09     564 1148.61   599.4 1148.56   619.8 1156.38
#Mann= 7, -1 ,  0
       0     0.1       0  283.46    0.06       0   305.6   0.045       0
  322.25    0.06       0   403.5    0.07       0     526    0.06       0
     596    0.05       0
Bank Sta=305.6,322.25
XS Rating Curve= 0 ,0
Exp/Cntr(USF)=0,0
Exp/Cntr=0.3,0.1

Type RM Length L Ch R = 1 ,22002   ,313.8,312.2,310.5
XS GIS Cut Line= 6
1680315.96469517423270.463140249  1680392.625303423324.427599251
1680525.50233383423417.9657980051680607.26332517423475.543110669
1680740.14330876423569.0832779261680816.80424467423623.048065007
#Sta/Elev= 30
       0 1166.89    63.8 1166.55    96.3 1164.59   117.6 1161.14   151.8 1152.33
   184.3 1141.64   193.9 1136.65   231.3 1122.02   254.2 1107.79   264.3 1103.26
   274.1 1094.42   280.1 1090.05   288.8 1084.67   294.4 1082.35   308.4 1080.81
  314.871082.435   323.1 1085.66     415 1085.97   420.9 1088.43   429.3 1094.05
   434.4 1096.23   452.3 1099.89   464.9 1107.93   469.2 1109.77   499.1 1112.64
     504  1116.1   513.8  1125.5   528.5 1130.38   552.5 1140.87   612.5 1161.36
#Mann= 5, -1 ,  0
       0     0.1       0   294.4   0.045       0  314.87     0.1       0
  406.25    0.06       0  518.75     0.1       0
Bank Sta=294.4,314.87
XS Rating Curve= 0 ,0
Exp/Cntr(USF)=0,0
Exp/Cntr=0.3,0.1

Type RM Length L Ch R = 1 ,21690   ,323,321.6,319.1
XS GIS Cut Line= 2
1680189.76730473  423606.87074391680732.68142574423875.254705608
#Sta/Elev= 30
       0 1190.31    38.3 1173.41    87.4 1159.97   122.4 1146.22   149.9 1130.09
   185.6 1112.72   211.4 1094.93   226.9 1080.14   230.2 1078.77   234.6 1078.63
   244.9 1078.82  249.96 1080.24   256.8 1081.62   307.6 1081.79   328.3 1084.31
   349.4 1084.94   355.1  1086.1     373 1093.43   390.8 1106.03   399.7 1107.54
   417.6 1107.26   426.5 1117.47     431 1121.03   439.9 1125.87   444.4 1127.32
   457.7 1128.27   471.1 1135.15   486.8 1140.82   529.1 1153.67   605.6 1169.48
#Mann= 5, -1 ,  0
       0     0.1       0   226.9   0.045       0  249.96     0.1       0
     290    0.06       0     400     0.1       0
Bank Sta=226.9,249.96
XS Rating Curve= 0 ,0
Exp/Cntr(USF)=0,0
Exp/Cntr=0.3,0.1

Type RM Length L Ch R = 1 ,21368   ,133.7,136.7,139.6
BEGIN DESCRIPTION:
Structure 8 XS 4
END DESCRIPTION:
XS GIS Cut Line= 3
1680033.39648318424040.5673712161680208.20589752423975.642599682
1680614.51054801424112.542410349
#Sta/Elev= 30
       0 1156.69    23.9 1152.25    39.5 1147.28    49.8 1139.51    66.9 1131.18
    86.1 1118.43   109.6 1105.58   122.4 1092.94   129.7 1089.21   194.8 1090.77
   203.3 1089.88   232.8 1082.67   308.8 1081.76   319.7 1077.98   331.3 1076.97
   342.6 1075.77     351 1076.91   372.1 1081.41   376.3 1084.17   392.3 1099.64
   397.4 1102.17   422.8 1101.32   435.4 1112.34   442.8 1115.93   455.5 1118.43
   486.1 1129.52     503 1132.26   532.5 1140.61   578.6 1146.42   615.2 1148.93
#Mann= 7, -1 ,  0
       0     0.1       0     130    0.06       0  236.48     0.1       0
   331.3   0.045       0     351     0.1       0  356.48    0.06       0
  436.48     0.1       0
Bank Sta=331.3,351
XS Rating Curve= 0 ,0
Exp/Cntr(USF)=0,0
Exp/Cntr=0.3,0.1

Type RM Length L Ch R = 1 ,21231   ,42.4,43.2,43
BEGIN DESCRIPTION:
Structure 8 XS 3
END DESCRIPTION:
XS GIS Cut Line= 6
1679998.21081298424189.7351492881680236.88815297424094.469086545
1680274.78970481424133.3950046551680340.34914584424184.613317958
1680348.54407597424211.2468408761680581.07521837424197.930079417
#Sta/Elev= 30
       0 1180.17    36.5 1168.58    83.9 1160.92    96.8 1156.21   139.9 1127.07
   148.5 1122.66   165.7 1109.32   196.3 1082.77     301  1080.7   317.5 1079.61
   323.7 1076.54   332.6 1074.91   344.5 1076.63   351.9 1080.48   357.1 1081.28
   422.6 1081.79   430.2 1084.53   438.2 1090.04   446.2 1092.34   470.3 1091.13
   474.2 1093.11     483 1102.63   490.3 1107.71   502.3 1109.44     517 1116.29
   550.4 1124.06   606.5 1140.04   626.5 1140.85   638.5  1143.8   655.5 1144.47
#Mann= 5, -1 ,  0
       0     0.1       0   323.7   0.045       0   344.5     0.1       0
  422.59    0.06       0  522.59     0.1       0
Bank Sta=323.7,344.5
XS Rating Curve= 0 ,0
Exp/Cntr(USF)=0,0
Exp/Cntr=0.3,0.1

Type RM Length L Ch R = 1 ,21188   ,201,191.7,182.7
BEGIN DESCRIPTION:
Structure 8 XS 2
END DESCRIPTION:
XS GIS Cut Line= 6
1680008.45447564424218.4174047381680222.54702524424137.492469719
1680301.42322773424204.0762770131680316.78872172424224.563602334
1680322.93491932 424249.148392721680581.07521837  424225.5879686
#Sta/Elev= 30
       0 1177.64    38.1 1166.83    80.9 1160.88      98 1154.56   110.8 1146.35
   119.4 1138.37     145 1121.25   166.4 1100.67   192.1  1083.2   202.9 1081.71
   233.1  1081.1   276.7 1078.52  287.381076.207   297.5 1074.88   306.3 1074.94
   311.2 1076.16   320.4 1080.22     326 1080.82   410.9 1081.24   416.8 1082.49
   428.8 1089.01   432.8 1089.83   456.9 1088.89     461 1090.48     473 1102.26
     477 1104.45   517.6 1119.38   577.4 1133.63   597.5 1137.44   642.7 1141.86
#Mann= 5, -1 ,  0
       0     0.1       0  287.38   0.045       0   311.2     0.1       0
  413.46    0.06       0  513.46     0.1       0
Bank Sta=287.38,311.2
XS Rating Curve= 0 ,0
Exp/Cntr(USF)=0,0
Exp/Cntr=0.3,0.1

Type RM Length L Ch R = 1 ,20996   ,132.7,124.1,113.6
BEGIN DESCRIPTION:
Structure 8 XS 1
END DESCRIPTION:
XS GIS Cut Line= 6
1680001.39609858424456.1198896771680174.12869276424391.423824832
1680246.87362601424367.1725610051680345.85177451424351.018065751
1680507.75138509424337.0633692591680600.35553059 424321.06832251
#Sta/Elev= 30
       0 1207.91    24.3 1198.51    71.3 1177.01    92.7 1168.65     114 1161.61
   135.4 1157.47   147.8 1148.27   158.3  1145.9   169.5  1140.8     178 1130.62
   186.5 1125.23   203.4 1108.47   211.8 1102.96   226.2 1095.74   257.9 1086.61
   270.5 1084.79   286.7 1077.55  301.89 1074.88   315.1 1072.33   323.2 1074.81
   351.6 1076.43   371.7 1075.72   379.8 1077.29   391.8 1082.57   423.9 1082.84
     444 1088.07     460 1090.31   476.1 1097.04   528.3 1112.97   617.9 1131.08
#Mann= 5, -1 ,  0
       0     0.1       0  271.13    0.06       0  301.89   0.045       0
   323.2    0.06       0  466.42     0.1       0
Bank Sta=301.89,323.2
XS Rating Curve= 0 ,0
Exp/Cntr(USF)=0,0
Exp/Cntr=0.3,0.1

Type RM Length L Ch R = 1 ,20872   ,48.7,50.1,48.7
BEGIN DESCRIPTION:
Structure 7 XS 3
END DESCRIPTION:
XS GIS Cut Line= 6
1680051.47785881424501.1424941711680279.91153614424532.897848418
1680308.59379159424509.337424299 1680347.5197097424448.899814601
1680371.08013382424424.3150242161680620.00113648424431.485588078
#Sta/Elev= 30
       0 1184.07      37 1167.56    57.3 1160.71    77.5 1155.62   105.8 1142.89
   113.9  1134.6     126 1125.61   134.1 1116.69   146.2 1112.77   202.9  1086.9
     215 1078.17   281.8 1076.81   294.2 1074.53   302.2 1071.69   306.9 1071.36
   311.6 1071.58  319.131074.585   331.8 1077.33   386.9 1080.12   406.9 1079.23
   410.9 1080.01   414.9 1081.86   422.9  1087.7   434.9 1092.84   458.9 1105.53
   476.2 1111.24   527.1 1131.17   573.4 1145.35     591 1149.52   622.9  1154.6
#Mann= 5, -1 ,  0
       0     0.1       0   294.2   0.045       0  319.13     0.1       0
  337.92    0.06       0  453.86     0.1       0
Bank Sta=294.2,319.13
XS Rating Curve= 0 ,0
Exp/Cntr(USF)=0,0
Exp/Cntr=0.3,0.1

Type RM Length L Ch R = 1 ,20822   ,311,321.2,336.1
BEGIN DESCRIPTION:
Structure 7 XS 2
END DESCRIPTION:
XS GIS Cut Line= 6
1680041.23419615424528.8003833541680306.54505906424570.799400263
1680334.20294825424543.1415110791680363.90956996424494.996296574
1680385.42126155424466.3140411241680609.75747382424471.435872455
#Sta/Elev= 30
       0 1187.01    19.1 1177.45    43.4 1167.19    83.9 1156.06   116.3 1141.25
   124.4 1134.52   132.5 1122.83   136.6 1119.74   144.7 1115.92   152.8 1110.08
   160.9  1108.3   173.6 1100.25   198.1 1089.42   213.5 1079.14     250 1077.33
   268.6 1074.15   310.8 1074.73   320.2 1072.82   331.4 1070.86  344.431072.861
   366.2 1077.88     398 1079.35   418.9 1079.01   422.9 1081.01   438.9    1093
   486.6 1113.88     534 1133.05   578.9 1148.29   602.9 1154.13   624.5 1157.85
#Mann= 4, -1 ,  0
       0     0.1       0   320.2   0.045       0  344.43    0.06       0
  460.15     0.1       0
Bank Sta=320.2,344.43
XS Rating Curve= 0 ,0
Exp/Cntr(USF)=0,0
Exp/Cntr=0.3,0.1

Type RM Length L Ch R = 1 ,20501   ,490.3,498.9,508.6
BEGIN DESCRIPTION:
Structure 7 XS 1
END DESCRIPTION:
XS GIS Cut Line= 6
1679974.95356618424752.7925246661680064.96322867424779.406644672
1680149.69304609424801.2842255831680392.60988308424860.373346254
1680477.63071042424881.0537510961680568.72436026424903.212499425
#Sta/Elev= 30
       0 1173.79    30.4 1158.99    72.1 1143.15   109.5  1121.5   121.9 1115.38
   208.6 1077.37   229.1 1072.81     295 1070.66   303.2  1068.4   307.4 1068.38
   315.6 1070.61   327.9 1072.34   348.5 1084.13   351.6 1084.97     365 1085.85
   373.2 1084.61   377.3 1085.52   385.6 1090.07   406.2 1097.71   418.5 1104.92
   426.7 1106.85   431.1 1110.04     451 1120.19   455.6 1124.61   463.8 1137.39
   470.8 1141.85   487.4 1146.05   521.4 1159.71   558.5 1169.06   612.6 1188.64
#Mann= 5, -1 ,  0
       0     0.1       0  286.37    0.06       0     295   0.045       0
   315.6    0.06       0  386.37     0.1       0
Bank Sta=295,315.6
XS Rating Curve= 0 ,0
Exp/Cntr(USF)=0,0
Exp/Cntr=0.3,0.1
