HEC-RAS study SUGARRN.prj: SUGARRN

--- SUGARRN.g01 (geometry) --- (continued)

Type RM Length L Ch R = 1 ,20002   ,233.5,218.3,197.6
BEGIN DESCRIPTION:
Structure 6 XS 4
END DESCRIPTION:
XS GIS Cut Line= 6
1679847.76746884424929.9703199271679931.75877067425090.585156173
1680012.85342476425245.6612895881680123.97853059425271.875804082
1680243.15972267425297.0411080871680361.65456443425321.355035841
#Sta/Elev= 30
       0 1160.71    11.9 1153.85    22.9 1149.65    52.5 1142.19    69.8  1139.4
    75.1 1137.06    88.7 1125.76      97 1116.16   102.2 1111.88   151.9 1081.18
   165.4 1074.23   185.9 1069.17     197 1068.04   296.3 1066.89   307.4 1064.54
   318.9 1067.01   336.9 1068.63   400.7 1067.95   417.1 1074.35   425.4 1075.54
   434.5  1081.4   458.2 1080.41   462.3  1081.7   474.7 1091.17     491 1097.38
   507.4 1099.04   527.8 1107.17   560.5  1114.9   646.3 1142.83   713.2 1158.07
#Mann= 5, -1 ,  0
       0     0.1       0   296.3   0.045       0   318.9    0.05       0
  396.25    0.06       0  500.43     0.1       0
Bank Sta=296.3,318.9
XS Rating Curve= 0 ,0
Exp/Cntr(USF)=0,0
Exp/Cntr=0.3,0.1

Type RM Length L Ch R = 1 ,19784   ,31.8,31.8,31.7
BEGIN DESCRIPTION:
Structure 6 XS 3
END DESCRIPTION:
XS GIS Cut Line= 4
 1679734.9486826425472.2417143951679882.45742491425410.779738432
1679962.35799367425308.3431118261680345.47097717425333.952268477
#Sta/Elev= 30
       0 1142.05     5.6 1139.42    43.5 1115.47    53.3 1111.33    83.6 1102.73
   105.3  1091.9   126.9 1079.29   139.9 1073.96   156.7 1070.08   223.5 1067.23
   228.6 1066.53   233.7 1064.25   238.7 1062.98   248.9 1064.26   259.5 1067.59
   343.6 1067.66   379.7 1069.17   387.7 1070.59   399.7 1079.21   403.7  1080.5
   427.8  1078.3   431.8 1079.93   439.8 1087.87   463.9 1096.46   475.9 1102.47
   499.9 1104.44   514.8 1110.84   596.2 1132.65   616.2 1140.17   673.7  1155.1
#Mann= 9, -1 ,  0
       0     0.1       0      30    0.05       0     130    0.06       0
   169.8    0.05       0   233.7   0.045       0   248.9    0.05       0
   279.8     0.1       0  379.71    0.06       0  479.71     0.1       0
Bank Sta=233.7,248.9
XS Rating Curve= 0 ,0
Exp/Cntr(USF)=0,0
Exp/Cntr=0.3,0.1

Type RM Length L Ch R = 1 ,19752   ,235.6,242,245.6
BEGIN DESCRIPTION:
Structure 6 XS 2
END DESCRIPTION:
XS GIS Cut Line= 4
1679746.21671153425496.8265047811679899.87165144425441.510726413
1679976.69912139425341.1228323391680346.49534344425349.317762468
#Sta/Elev= 30
       0 1145.17    20.5 1134.27    48.8 1116.34    82.8 1103.25     104 1089.03
   133.8 1073.37   142.3 1071.16   163.3 1068.56   229.8 1067.94   241.2  1067.2
   250.2 1064.38   258.3  1062.6  265.661064.421   270.3 1066.42   280.4 1067.42
   361.2 1067.48   369.2  1070.3   381.2 1078.59   385.2 1079.71   413.2 1077.06
   417.2 1079.68   424.7 1088.92   428.8 1091.83   453.4 1099.01   465.2 1103.92
   489.2 1106.89   505.2 1112.91   561.2 1128.11   617.2 1146.05   659.6 1157.85
#Mann= 8, -1 ,  0
       0     0.1       0      20    0.05       0     120    0.06       0
  213.31    0.05       0   250.2   0.045       0  265.66     0.1       0
  369.72    0.06       0  469.72     0.1       0
Bank Sta=250.2,265.66
XS Rating Curve= 0 ,0
Exp/Cntr(USF)=0,0
Exp/Cntr=0.3,0.1

Type RM Length L Ch R = 1 ,19510   ,255.5,257.2,258.3
BEGIN DESCRIPTION:
Structure 6  XS 1
END DESCRIPTION:
XS GIS Cut Line= 3
1679816.89798389425619.7504567081680159.03631675425508.094533707
1680361.86083743425495.802138514
#Sta/Elev= 30
       0 1131.35      16 1115.51    20.2 1112.76    49.7 1102.06    83.3 1082.77
   100.2 1075.61   108.6 1070.67   116.1 1068.34   142.2 1065.44   287.3 1064.32
   297.9 1063.86   302.1  1062.2   309.6 1061.15     319  1062.2   327.4 1068.11
   331.6 1069.36   356.8 1071.81     361 1074.01     365 1078.46     373 1090.81
     377 1095.96     389 1109.45   421.1 1123.65   437.1 1125.51   441.1 1127.21
   445.1 1130.69   449.1 1132.81   533.3 1157.85   545.6 1160.66   563.1 1163.07
#Mann= 6, -1 ,  0
       0     0.1       0     150    0.05       0     250    0.06       0
   302.1   0.045       0     319    0.06       0   419.9     0.1       0
Bank Sta=302.1,319
XS Rating Curve= 0 ,0
Exp/Cntr(USF)=0,0
Exp/Cntr=0.3,0.1

Type RM Length L Ch R = 1 ,19253   ,171.5,172.3,173.4
BEGIN DESCRIPTION:
Structure 5 XS 4
END DESCRIPTION:
XS GIS Cut Line= 6
1679833.32441782425884.6917159261679927.99384792425839.102568254
1680014.78402866425799.8001534341680088.34621749425783.896641925
1680348.40770524425748.2008471791680441.28678458425735.452185005
#Sta/Elev= 30
       0 1149.99    20.9 1141.82    56.1 1120.36    71.1 1113.55      83 1110.23
   122.8  1093.2   144.7  1086.3   175.5 1074.42   197.4 1064.12     214 1062.28
   291.5 1061.82   303.6 1059.82   315.8 1058.57   322.11059.888   331.9 1065.45
   352.1 1063.94   356.1 1065.16   364.2 1073.64   376.3 1084.74   384.4 1090.86
   404.6 1099.63   428.8 1108.73   469.2  1129.3   489.4  1138.6   509.1 1146.12
   545.9 1156.57     562  1158.3   570.1 1160.94   594.4  1164.5   631.9 1172.04
#Mann= 5, -1 ,  0
       0     0.1       0   303.6   0.045       0   322.1     0.1       0
  345.61    0.06       0  445.61     0.1       0
Bank Sta=303.6,322.1
XS Rating Curve= 0 ,0
Exp/Cntr(USF)=0,0
Exp/Cntr=0.3,0.1

Type RM Length L Ch R = 1 ,19081   ,57.9,57.9,57.5
BEGIN DESCRIPTION:
Structure 5 XS 3
END DESCRIPTION:
XS GIS Cut Line= 3
1679867.07148519425948.1779706681679980.56881456425954.483062247
1680505.05539587425922.729055622
#Sta/Elev= 30
       0 1136.54    13.1 1130.92    49.1 1109.07    69.1 1104.52   105.2  1084.9
   117.2 1079.48   141.3 1071.11   149.3 1066.21   201.4 1062.59   285.5 1062.16
  299.79 1059.67   309.6 1056.08   313.6 1056.45  320.181059.687   325.6 1062.19
   349.6 1062.79   353.7 1064.12   361.7 1073.34   373.7 1084.27   389.7 1094.96
   402.3 1101.22   417.8 1110.72   481.9 1141.51   497.9 1150.39     538 1157.49
   554.7  1162.9   574.1 1164.43   606.1  1173.5   630.2 1178.27   639.1 1181.83
#Mann= 7, -1 ,  0
       0     0.1       0      90    0.06       0  193.67     0.1       0
  283.67    0.06       0  299.79   0.045       0  320.18    0.06       0
  383.67     0.1       0
Bank Sta=299.79,320.18
XS Rating Curve= 0 ,0
Exp/Cntr(USF)=0,0
Exp/Cntr=0.3,0.1

Type RM Length L Ch R = 1 ,19023   ,512.7,520.9,524.6
BEGIN DESCRIPTION:
Structure 5 XS 2
END DESCRIPTION:
XS GIS Cut Line= 3
1679858.92748967426005.1793937541679972.42481904426011.484485333
1680496.91140035425979.730478709
#Sta/Elev= 30
       0 1152.26     9.2 1150.23    21.2 1144.74    52.8 1123.59    65.3 1118.07
   101.3 1095.75   117.4 1087.73   129.4 1079.83   141.4 1068.81   145.4 1066.34
   177.5 1063.48   201.5 1063.14   221.6 1061.38   253.6 1060.21   317.7 1060.77
     324 1059.46   333.8 1056.27  342.561059.478   345.8 1061.06   354.2 1062.41
   373.8 1063.11   401.9 1083.43     450 1113.33     466 1120.89   542.1 1151.94
   554.5 1156.32   578.2 1162.45   594.2 1164.23   610.3 1170.92   639.1 1178.91
#Mann= 5, -1 ,  0
       0     0.1       0  293.67    0.06       0     324   0.045       0
  342.56    0.06       0  393.67     0.1       0
Bank Sta=324,342.56
XS Rating Curve= 0 ,0
Exp/Cntr(USF)=0,0
Exp/Cntr=0.3,0.1

Type RM Length L Ch R = 1 ,18502   ,499.9,500,499.4
BEGIN DESCRIPTION:
Structure 5 XS 1
END DESCRIPTION:
XS GIS Cut Line= 6
 1679706.4278565426235.5408715011679784.43294984426287.544048339
1680002.84557076426433.1533371661680064.84150976426475.367491588
1680126.90897092426539.7869821791680192.80811734426612.980077252
#Sta/Elev= 30
       0 1227.33    21.3 1218.16    35.7 1208.09    45.3 1200.06   107.8 1166.74
   122.2 1160.89   160.6 1150.61   182.1 1139.88     201  1132.1   213.6 1125.11
   242.4 1106.56   252.9 1095.23   261.5 1087.94   271.2 1076.41   281.7 1066.14
   293.3 1056.74   297.5 1054.49   300.1 1053.45   309.7 1053.18  317.521054.528
   328.9 1056.61   385.5 1057.26   420.7  1059.9   460.7 1059.61   499.4 1062.65
   541.9 1080.54   561.7 1094.23   594.2 1114.24   613.2 1117.72   619.2 1122.35
#Mann= 5, -1 ,  0
       0     0.1       0   297.5   0.045       0  317.52     0.1       0
  416.25    0.06       0  560.71     0.1       0
Bank Sta=297.5,317.52
XS Rating Curve= 0 ,0
Exp/Cntr(USF)=0,0
Exp/Cntr=0.3,0.1

Type RM Length L Ch R = 1 ,18002   ,504.2,501,492.4
XS GIS Cut Line= 6
1679442.57963093426663.6203959291679521.50598225426714.213798672
1679595.17020501426761.4345047621679805.64025651426896.350901589
1679879.30480734426943.5712795851679958.23083059426994.165010422
#Sta/Elev= 30
       0  1147.8    46.2  1143.1    82.6 1137.14   101.6 1132.85   134.9 1123.38
   218.9 1092.26   229.9 1090.04   250.8 1083.87   253.7 1082.31   277.4 1061.16
  294.921047.887   297.1 1046.92   301.2 1046.64   310.7 1046.88   314.5 1047.78
   320.4 1050.19   324.9  1050.8   362.9 1052.05   377.2 1053.83   400.9 1054.94
     410 1058.85   412.9 1059.27   434.2 1058.52   446.4 1069.84   462.7 1078.97
   476.1 1083.42   500.7 1094.48   567.2 1119.04   583.7 1124.58   612.5  1132.1
#Mann= 5, -1 ,  0
       0     0.1       0  294.92   0.045       0   314.5     0.1       0
  406.25    0.06       0  588.75     0.1       0
Bank Sta=294.92,314.5
XS Rating Curve= 0 ,0
Exp/Cntr(USF)=0,0
Exp/Cntr=0.3,0.1

Type RM Length L Ch R = 1 ,17501   ,500.3,500.6,500.4
XS GIS Cut Line= 6
1679180.04669142427254.7661952531679361.22119784427259.992890835
  1679436.190208427262.1552880851679611.11735159427267.201537833
1679698.58108743427269.724498674  1679792.429653427269.913474679
#Sta/Elev= 30
       0 1219.58    36.1 1200.43    56.1 1191.58    68.1 1184.58    80.1 1180.84
    96.1 1170.49   128.1 1152.25   144.1  1147.9   163.1 1138.76   200.2 1113.34
   220.2 1102.47   244.2 1086.13   260.2 1077.02   264.2 1072.91   272.2 1066.63
   280.2 1057.26  298.391044.709   300.2 1043.57   308.2 1043.04   320.2 1044.48
   336.2 1045.72   356.3 1049.28   416.2 1050.41   444.3 1049.78   468.3 1051.56
   484.1  1054.8   508.3 1054.09   520.3 1062.13   544.3 1076.39   612.6 1105.36
#Mann= 5, -1 ,  0
       0     0.1       0  286.25    0.06       0  298.39   0.045       0
   320.2    0.06       0  578.75     0.1       0
Bank Sta=298.39,320.2
XS Rating Curve= 0 ,0
Exp/Cntr(USF)=0,0
Exp/Cntr=0.3,0.1

Type RM Length L Ch R = 1 ,17000   ,502.9,499.9,496.4
XS GIS Cut Line= 6
1679193.50466976427713.8440172521679287.96182993427732.651066259
1679376.27562967427749.1444715861679451.97921842427760.372467503
1679551.93800801427763.9393895121679808.26951633427756.257646337
#Sta/Elev= 30
       0 1090.59    27.1 1087.74    92.4 1077.43   116.8 1071.91     129 1067.19
   133.1 1066.36   153.4 1065.28   181.7 1058.29   198.1 1047.84   206.2 1044.93
   250.7 1043.25   290.8 1043.58   294.8  1042.8  300.871040.227   314.9 1039.38
   322.9 1040.17   332.5 1045.09   342.9  1048.8   354.9 1049.02   370.9 1048.04
   378.9 1053.14   386.9 1060.48   410.9 1076.22   428.3 1085.73   450.9 1096.13
   470.9 1106.35   498.9 1117.51     545 1138.04     579 1149.09   619.2 1158.15
#Mann= 5, -1 ,  0
       0     0.1       0  272.68    0.06       0  300.87   0.045       0
   322.9    0.06       0  372.71     0.1       0
Bank Sta=300.87,322.9
XS Rating Curve= 0 ,0
Exp/Cntr(USF)=0,0
Exp/Cntr=0.3,0.1

Type RM Length L Ch R = 1 ,16500   ,268.2,263.5,258.3
XS GIS Cut Line= 6
1679199.27467135428311.5977430051679376.47313584428273.490535751
1679449.79680809428257.7218665031679620.88537668428220.928961083
1679706.42949693428202.5320162621679798.08416925428182.821753845
#Sta/Elev= 30
       0 1168.22      50    1155    78.6  1145.1      95  1140.8   131.8 1128.05
   158.7 1117.66   209.5 1096.03   242.3 1079.21   262.6 1060.26   266.8 1052.52
   270.9 1046.99   279.4 1040.35   289.5 1037.15   299.4 1036.09   316.4 1037.04
   328.2 1039.31   360.9 1039.46   385.5 1042.08   401.8 1041.58   417.5 1044.24
   434.6 1049.04   459.1 1063.01   471.4 1074.08   474.7 1076.23   492.3 1079.59
   516.4 1096.42   524.6  1099.9   557.3 1116.98   575.7 1123.99   612.5 1135.46
#Mann= 5, -1 ,  0
       0     0.1       0  276.25    0.06       0   289.5   0.045       0
   316.4    0.06       0  471.25     0.1       0
Bank Sta=289.5,316.4
XS Rating Curve= 0 ,0
Exp/Cntr(USF)=0,0
Exp/Cntr=0.3,0.1

Type RM Length L Ch R = 1 ,16237   ,129.6,131.3,134
BEGIN DESCRIPTION:
Structure 4 XS 4
END DESCRIPTION:
XS GIS Cut Line= 5
1679348.70080376428467.3506782761679529.58339902428512.986195429
1679583.51628293428499.7104086211679613.38680325428478.137255058
1679874.75385603428402.631217586
#Sta/Elev= 30
       0 1127.38    57.1 1110.44    69.5 1105.27    94.3  1093.5   114.9 1085.51
   123.2 1080.87   139.7 1070.03   180.9 1045.44   193.3 1038.65   201.5 1037.78
   238.6 1037.06   250.5 1034.88     262 1034.01  271.441034.915   294.3 1038.07
   315.1 1039.26   331.7 1039.05   335.9 1040.74   340.1 1045.04     347 1058.12
   350.3 1062.32   369.2  1080.6   377.5 1085.31   385.9 1088.11   411.6 1098.75
   423.3 1102.55     465 1110.44   523.3 1128.26   535.8 1130.41     551 1134.43
#Mann= 5, -1 ,  0
       0     0.1       0   250.5   0.045       0  271.44     0.1       0
  328.94    0.06       0  358.94     0.1       0
Bank Sta=250.5,271.44
XS Rating Curve= 0 ,0
Exp/Cntr(USF)=0,0
Exp/Cntr=0.3,0.1

Type RM Length L Ch R = 1 ,16105   ,38.6,38.8,38.8
BEGIN DESCRIPTION:
Structure 4 XS 3
END DESCRIPTION:
XS GIS Cut Line= 6
1679376.08211405428766.0558814591679485.60735522428714.612207578
1679567.75128609428634.9574867291679596.79206974428622.511436596
1679616.70574995 428612.554596491679974.32225709428518.794352158
#Sta/Elev= 30
       0  1082.9    13.3 1080.52    26.6 1076.06    46.3 1067.86    61.9 1059.08
      84 1049.46    97.4 1045.86   138.4 1042.59   227.4 1038.88   292.8 1037.37
   334.2 1037.77  340.03 1034.36   342.4 1032.83   346.6 1032.18   351.61034.218
   354.8 1036.71     359  1038.1   387.9 1038.34   392.1 1039.74   396.2 1043.64
   404.5 1058.77   408.6 1061.91   431.3    1075   449.9  1082.2   507.8 1098.44
   541.1    1106   573.8 1115.68     589 1119.14   615.4 1122.72     659 1125.64
#Mann= 5, -1 ,  0
       0     0.1       0  231.01    0.06       0  340.03   0.045       0
   351.6    0.06       0  439.29     0.1       0
Bank Sta=340.03,351.6
XS Rating Curve= 0 ,0
Exp/Cntr(USF)=0,0
Exp/Cntr=0.3,0.1

Type RM Length L Ch R = 1 ,16067   ,261.3,261.1,260.5
BEGIN DESCRIPTION:
Structure 4 XS 2
END DESCRIPTION:
XS GIS Cut Line= 6
1679387.69842751428792.607455075 1679499.7128787428733.696151114
1679553.64576261428680.5930038821679599.28127976428654.871166941
1679653.21416367428642.4251168081679979.30067715428562.770395959
#Sta/Elev= 30
       0 1090.91    12.2 1089.74    18.5 1087.99      30 1082.82    54.7 1069.71
    86.3 1054.33    98.1 1049.18   108.9 1046.41   136.2 1043.05     151 1042.08
   320.6 1035.73   329.4 1034.64   333.8 1032.48   337.7 1031.08   341.8 1031.03
  346.661032.458   354.1 1037.92   378.9 1039.03     383 1043.19   391.2 1059.69
   395.3 1065.15   403.3 1073.07   407.7 1076.68   424.1 1086.05   461.2 1099.89
   539.4 1122.44   556.5  1126.3   589.2  1131.6   617.7 1134.36   645.7 1135.81
#Mann= 5, -1 ,  0
       0     0.1       0  212.25    0.06       0   333.8   0.045       0
  346.66    0.06       0  419.99     0.1       0
Bank Sta=333.8,346.66
XS Rating Curve= 0 ,0
Exp/Cntr(USF)=0,0
Exp/Cntr=0.3,0.1

Type RM Length L Ch R = 1 ,15805   ,305.9,305.4,304.7
BEGIN DESCRIPTION:
Structure 4 XS 1
END DESCRIPTION:
XS GIS Cut Line= 2
1679428.39785731428967.9252936241680036.02034366428813.336178468
#Sta/Elev= 30
       0 1138.46    16.2 1131.21    28.6  1128.4    49.2 1117.31    81.5 1096.26
   111.1 1078.46   148.3 1049.74   160.7 1042.25   168.9 1038.78   173.7 1037.48
   185.4  1036.6   288.6 1033.47   296.9 1031.34   305.3 1030.15     316 1031.23
   325.8  1035.4   350.5 1036.26   354.7 1039.55   358.8  1046.8     367 1063.86
   371.2 1069.03   384.2 1080.53   391.8 1085.61   410.6 1091.85   433.6 1100.98
   474.4 1113.63   532.3 1138.33     561 1148.68   577.5 1153.89     627 1164.44
#Mann= 5, -1 ,  0
       0     0.1       0     240    0.06       0   296.9   0.045       0
     316    0.06       0     340     0.1       0
#XS Ineff= 2 , 0
                          339.68         1063.59
Permanent Ineff=
       F       F
Bank Sta=296.9,316
XS Rating Curve= 0 ,0
Exp/Cntr(USF)=0,0
Exp/Cntr=0.3,0.1

Type RM Length L Ch R = 1 ,15500   ,503,500.7,495.5
XS GIS Cut Line= 6
 1679509.4659801429282.700459585 1679681.8022496 429226.56015192
1679753.11378676429203.3292272541679848.19594568429172.355535924
1679919.50748284429149.1246112591680091.84375234  429092.9839755
#Sta/Elev= 30
       0 1166.48    19.6 1154.73    32.4 1151.34    49.1 1145.12    61.7 1136.83
   116.4 1104.29     153 1083.56   175.5 1068.91   204.7 1046.53   221.5 1036.94
     230 1033.72   246.8 1030.74   288.9 1031.26  296.041028.542   305.3 1027.35
   314.1 1028.53   322.5 1032.36   326.7 1033.14   352.9 1033.45   360.4 1039.37
   371.9 1054.25   385.6 1066.73   403.6 1079.79   416.3 1086.33   448.1 1099.78
   486.6 1113.07   536.9 1136.72   559.1 1145.65   566.5 1148.44   612.5 1160.43
#Mann= 5, -1 ,  0
       0     0.1       0  266.25    0.06       0  296.04   0.045       0
   314.1    0.06       0  366.25     0.1       0
Bank Sta=296.04,314.1
XS Rating Curve= 0 ,0
Exp/Cntr(USF)=0,0
Exp/Cntr=0.3,0.1

Type RM Length L Ch R = 1 ,14999   ,488.8,497.8,510.3
XS GIS Cut Line= 6
1679667.09033675429842.5379225911679876.75231901429695.208820924
1679958.57203725429637.7148414251680029.83337767429594.200820833
1680114.30729009429543.0332722511680202.49740243429488.257791251
#Sta/Elev= 30
       0 1192.39    22.3 1183.82    45.2 1171.19    69.7 1160.61      87 1154.15
   103.9 1149.35   121.8    1137   163.5 1111.88   219.2 1080.81   272.1 1041.39
   280.7 1034.02   289.3 1029.98     295 1025.94   303.6 1024.83     318 1025.96
   338.1 1027.79   381.5 1027.25   395.6 1030.68   404.6 1031.31   428.1 1029.93
     433 1033.23   442.6 1043.96   451.8 1051.25   489.2  1070.8   509.6 1076.98
   535.9 1081.78   573.6 1085.79   605.5 1083.02   626.6 1083.18   642.3 1081.92
#Mann= 5, -1 ,  0
       0     0.1       0     295   0.045       0     318     0.1       0
  356.25    0.06       0  548.51     0.1       0
#XS Ineff= 2 , 0
                          411.14         1068.72
Permanent Ineff=
       F       F
Bank Sta=295,318
XS Rating Curve= 0 ,0
Exp/Cntr(USF)=0,0
Exp/Cntr=0.3,0.1

Type RM Length L Ch R = 1 ,14502   ,500.5,500.2,498.4
XS GIS Cut Line= 6
1679825.67663376430014.4660564211679932.82799426430003.132089585
1680020.12243909430021.8433382511680091.37459317430045.656938925
1680184.22250459430082.7953160851680422.14492901430177.963104755
#Sta/Elev= 30
       0 1152.92    10.5 1149.13    38.7 1129.32    90.9 1096.66     107 1088.19
   131.6 1080.41   172.7 1052.99   218.1 1027.23   226.5  1024.6   302.6 1025.29
   311.9  1021.8   320.3 1020.96   333.8 1021.74   344.5 1026.48   372.2 1028.24
   389.3 1043.03   402.2 1060.62   406.5 1068.29   410.8 1073.13   419.4 1080.32
   423.7 1082.96   466.8 1100.56   508.8 1123.59   522.8 1127.91     558 1151.75
   565.9  1154.5   582.7  1156.6   601.1 1162.34   617.6 1165.62   628.4 1169.66
#Mann= 5, -1 ,  0
       0     0.1       0   311.9   0.045       0   333.8     0.1       0
  342.15    0.06       0  442.15     0.1       0
Bank Sta=311.9,333.8
XS Rating Curve= 0 ,0
Exp/Cntr(USF)=0,0
Exp/Cntr=0.3,0.1

Type RM Length L Ch R = 1 ,14001   ,518.3,502.9,486.8
XS GIS Cut Line= 6
  1679684.736955430446.8296930041679930.18003367   430520.463404
1680025.96265051430549.1979265961680098.31388375 430569.03482917
1680183.56666601430589.3684499261680275.26989467430609.949773595
#Sta/Elev= 30
       0 1183.58    36.9 1161.49    49.5 1155.37    70.3 1148.07    95.4  1133.7
   112.1 1126.09   116.3  1123.2   124.6 1111.07   137.2 1103.53   171.1 1085.35
   212.3 1067.98     229  1054.4   245.7 1038.36   266.6 1023.61   291.7 1016.46
     306 1016.06  314.241016.471   350.1 1024.03   366.8 1024.12   375.1 1022.32
   379.2 1023.69   391.7 1032.66   408.3 1041.18   432.4  1050.8   457.8 1064.17
     466 1067.22   486.6  1070.9   519.5 1081.67   544.1 1095.06   612.9 1128.52
#Mann= 5, -1 ,  0
       0     0.1       0  286.25    0.06       0   291.7   0.045       0
  314.24    0.06       0  386.25     0.1       0
Bank Sta=291.7,314.24
XS Rating Curve= 0 ,0
Exp/Cntr(USF)=0,0
Exp/Cntr=0.3,0.1

Type RM Length L Ch R = 1 ,13498   ,495.1,499.1,502.7
XS GIS Cut Line= 6
1679931.21284001431245.6998144241680060.32872351 431024.35544084
1680110.71576184430937.9776608351680147.93845643430872.863289759
1680201.40586917430801.2541810131680281.19048651430738.660146087
#Sta/Elev= 30
       0 1156.08     9.7 1150.65    30.8 1141.63      43 1138.99    52.3 1132.89
    70.8 1113.79    80.1 1096.45    84.7 1089.89    98.6 1075.14   112.6  1064.2
   154.2 1049.48     177 1040.15   194.5 1025.33   205.1 1018.17   228.3 1015.15
   282.3 1014.68   293.1 1013.11   297.7 1011.66     307 1011.32   317.4 1013.03
   329.1 1020.41   334.9 1022.22   367.1 1021.81   375.2 1026.48   383.2 1032.73
   390.6 1036.18   422.4 1040.08   477.3 1056.19   560.7 1084.65     622 1111.38
#Mann= 5, -1 ,  0
       0     0.1       0  241.25    0.06       0   293.1   0.045       0
   317.4    0.06       0  441.25     0.1       0
Bank Sta=293.1,317.4
XS Rating Curve= 0 ,0
Exp/Cntr(USF)=0,0
Exp/Cntr=0.3,0.1

Type RM Length L Ch R = 1 ,12999   ,484.7,497.4,509.7
XS GIS Cut Line= 6
1680236.02751909431488.2977544221680432.03532918431323.237060919
  1680508.262867431258.510484338 1680563.2411035431207.361964583
1680627.53001693431147.679341167 1680697.3274495431084.601383343
#Sta/Elev= 30
       0 1152.23      34 1142.32    45.3 1140.08    86.6 1119.62   153.2 1080.15
   181.3 1067.77   215.6  1044.5   230.2 1037.45   238.4 1030.46     248  1020.3
   258.2  1012.8   266.8  1010.3     279 1009.81   293.1 1007.35   308.8 1006.53
   314.1 1007.33   322.2 1011.99   326.3 1012.68   343.4 1012.51   351.9 1014.15
   399.8 1012.28   419.8 1013.48   425.5 1015.84   436.8 1023.09   467.9 1051.32
   482.5 1062.19   494.3 1068.18   547.6 1082.08   569.8 1085.61   613.1  1089.4
#Mann= 5, -1 ,  0
       0     0.1       0  276.25    0.06       0   293.1   0.045       0
   314.1    0.06       0  406.25     0.1       0
Bank Sta=293.1,314.1
XS Rating Curve= 0 ,0
Exp/Cntr(USF)=0,0
Exp/Cntr=0.3,0.1

Type RM Length L Ch R = 1 ,12502   ,505.5,500.9,494.8
XS GIS Cut Line= 6
  1680290.826294431630.7587555941680391.42058101431649.714754418
1680480.19960292431675.2461994291680543.00557968431716.349463671
1680756.60882701431868.9272425031680832.89607601431923.418603346
#Sta/Elev= 30
       0 1123.27    66.4 1079.52    78.6  1072.2    94.9 1065.12   107.2  1055.3
   115.6 1051.55   144.7 1029.29   160.2 1014.59   169.7 1009.38   273.6 1008.57
   300.7 1006.95  310.141003.473   320.3 1001.52   328.1 1003.44   336.7 1008.54
   354.7 1009.58     374 1014.35   387.1 1025.58   403.9  1044.8   414.1 1061.71
   418.6 1066.78   465.7 1091.16   492.4 1108.03   502.2 1116.74   517.3  1126.6
   551.4 1143.44   571.8 1148.85   585.8 1149.97   614.2 1156.28   626.1 1160.42
#Mann= 5, -1 ,  0
       0     0.1       0  254.74    0.06       0  310.14   0.045       0
   328.1    0.06       0   429.8     0.1       0
Bank Sta=310.14,328.1
XS Rating Curve= 0 ,0
Exp/Cntr(USF)=0,0
Exp/Cntr=0.3,0.1

Type RM Length L Ch R = 1 ,12001   ,435.4,437.2,439.1
XS GIS Cut Line= 6
1680069.09314168432150.1100790951680161.97747034432162.820355505
1680248.66955417 432174.683192671680422.05372185432198.409195095
1680496.36131601432208.5771537571680675.93772851432233.150923505
#Sta/Elev= 30
       0 1181.15    23.2 1170.92    51.5    1153    79.8  1139.1    99.9 1134.46
   144.4 1106.46   196.8  1071.6     213 1064.08   233.2 1056.91   245.3  1046.2
   257.4  1031.2   273.5 1015.17   293.7  999.43   301.8  998.08     318  999.47
   362.4 1004.97   382.6  1005.8   394.7 1003.83   398.7 1005.38   410.8 1016.81
   451.2 1045.84   463.3 1055.99   479.4 1059.73   491.6 1066.96   507.7 1074.03
   515.8 1076.17   527.9  1082.7   541.1  1091.1   592.5 1129.77   612.5 1142.56
#Mann= 5, -1 ,  0
       0     0.1       0  286.25    0.06       0   293.7   0.045       0
     318    0.06       0  386.25     0.1       0
#XS Ineff= 2 , 0
                          384.47         1052.16
Permanent Ineff=
       F       F
Bank Sta=293.7,318
XS Rating Curve= 0 ,0
Exp/Cntr(USF)=0,0
Exp/Cntr=0.3,0.1

Type RM Length L Ch R = 1 ,11564   ,192.6,190.2,187.5
BEGIN DESCRIPTION:
Structure 3 XS 4
END DESCRIPTION:
XS GIS Cut Line= 6
1679983.45900198432520.5249086571680157.13614807432572.369293164
1680324.82446099432622.4256234871680396.69111515432643.877352248
1680480.11483282432670.6919311541680569.78328865432699.759130235
#Sta/Elev= 30
       0 1148.82      28 1136.69    59.1 1127.46    71.6 1121.91   100.9 1101.28
   125.9 1086.44   142.6 1073.64   159.3 1063.37   184.4 1053.29   212.7    1039
   259.5 1001.54   267.8  999.02   299.5  999.52   309.6  996.92     322  995.25
   334.9  996.99   351.3 1002.08   363.9  1002.5   376.4 1000.13   399.2 1011.55
   434.5  1036.3     444 1045.63   463.1 1059.83   506.3 1079.39   520.3 1089.69
   535.7 1092.82   548.9 1106.79   556.7 1113.08   598.8 1137.65   613.1 1140.88
#Mann= 5, -1 ,  0
       0     0.1       0  276.25    0.06       0   309.6   0.045       0
   334.9    0.06       0  386.25     0.1       0
Bank Sta=309.6,334.9
XS Rating Curve= 0 ,0
Exp/Cntr(USF)=0,0
Exp/Cntr=0.3,0.1

Type RM Length L Ch R = 1 ,11374   ,57.9,57.6,57.4
BEGIN DESCRIPTION:
Structure 3 XS 3
END DESCRIPTION:
XS GIS Cut Line= 3
1679990.04602635432585.8888535811680206.30112696432790.762106793
1680542.69795013 432829.96624784
#Sta/Elev= 30
       0 1118.27    27.1 1105.96    79.7 1085.85   113.7 1066.15   155.1 1049.08
   190.1 1022.73   221.2 1002.86   239.8  999.38   283.9  998.41   311.8 1001.51
  320.89997.1692   327.9  994.16     344  993.94   351.6  997.15   360.1 1002.65
   384.3 1002.45   388.3 1003.93   404.4 1022.05   424.6 1036.43   452.7 1061.53
     497 1074.52   513.2 1082.46   537.3  1097.2   553.4 1103.37   561.5 1104.07
   573.6 1108.42   597.7 1125.53   609.8 1127.87   621.9 1134.73   636.6 1137.64
#Mann= 4, -1 ,  0
       0     0.1       0  297.89    0.07       0  320.89   0.045       0
   351.6     0.1       0
Bank Sta=320.89,351.6
XS Rating Curve= 0 ,0
Exp/Cntr(USF)=0,0
Exp/Cntr=0.3,0.1

Type RM Length L Ch R = 1 ,11316   ,322.6,316.2,309.6
BEGIN DESCRIPTION:
Structure 3 XS 2
END DESCRIPTION:
XS GIS Cut Line= 3
1679967.28233154432604.8585992491680201.24252811432848.935993508
1680535.11005187432880.552236287
#Sta/Elev= 30
       0 1110.68    31.5 1097.09    68.3 1083.76    99.4 1067.91   149.2 1052.08
   192.7 1024.88   232.4 1002.79     260 1001.25     349  998.52     353  998.08
   361.1  993.72   369.1  992.66   386.8993.6885   388.1  994.28   401.3 1002.66
   425.4 1002.47   433.4 1005.47   437.4 1011.81   441.4 1020.38   453.5 1035.85
   461.5  1048.2   473.6 1058.39   532.6 1075.64     574 1098.13   606.2 1110.79
   622.2 1114.02   638.3 1124.21   646.3 1126.45   662.4 1135.27   673.5 1138.03
#Mann= 5, -1 ,  0
       0     0.1       0     260    0.07       0   361.1   0.045       0
   386.8    0.07       0   388.1     0.1       0
Bank Sta=361.1,386.8
XS Rating Curve= 0 ,0
Exp/Cntr(USF)=0,0
Exp/Cntr=0.3,0.1

Type RM Length L Ch R = 1 ,11000   ,490.6,498.6,505.4
BEGIN DESCRIPTION:
Structure 3 XS 1
END DESCRIPTION:
XS GIS Cut Line= 6
1679985.03589509433275.8197699191680071.82049842433240.359210923
1680314.81837201433141.0700394211680384.24638276433112.701329753
1680465.24589267433079.6059235041680551.81724185433043.623055846
#Sta/Elev= 30
       0 1100.28    24.9 1084.62    38.6 1071.69    55.2 1058.94      80 1044.68
    89.7 1036.31    98.4 1026.55     107 1020.38   128.6 1010.36   154.6 1004.16
   167.5  997.37   279.9  996.73   284.2  996.48   290.2  993.68   296.3   991.4
   301.5  991.04   310.1  991.27   317.8  993.56   327.4 1000.31   331.7 1001.75
   363.8 1002.36   385.3 1018.58   409.5 1030.24   425.1 1044.44   439.7 1053.04
     457 1060.71   474.3 1065.83   513.2 1088.21   526.2 1093.78   612.5 1109.24
#Mann= 7, -1 ,  0
       0     0.1       0      80    0.06       0  181.25    0.05       0
  286.25    0.06       0   290.2   0.045       0   317.8    0.06       0
  396.25     0.1       0
Bank Sta=290.2,317.8
XS Rating Curve= 0 ,0
Exp/Cntr(USF)=0,0
Exp/Cntr=0.3,0.1

Type RM Length L Ch R = 1 ,10501   ,502.7,500.4,498.4
XS GIS Cut Line= 6
1680028.58633292433557.0816745911680118.27086484433584.989099085
1680275.46871318433626.1606046711680372.20605251 433651.49684009
  1680444.759057433670.4987705951680620.09499243  433716.4196105
#Sta/Elev= 30
       0 1104.51    49.8 1084.95    66.5 1071.56    79.1 1068.46    91.7 1061.53
   116.5 1054.17   124.8 1050.16     133 1043.33   147.5 1027.62   186.8  992.31
   195.1  990.64   277.8   991.7   294.3  988.76   306.7  987.88   313.5988.7543
   323.3  992.38   360.5  994.22     377  998.41   397.7  997.69   414.2 1011.15
   430.8 1017.12   443.2 1024.49   480.4 1054.03   509.3 1071.61   518.9 1080.95
   527.6 1087.49   538.3 1093.15   550.7 1097.69     580 1114.81   612.7 1131.85
#Mann= 5, -1 ,  0
       0     0.1       0   294.3   0.045       0   313.5     0.1       0
  336.43    0.06       0  441.43     0.1       0
Bank Sta=294.3,313.5
XS Rating Curve= 0 ,0
Exp/Cntr(USF)=0,0
Exp/Cntr=0.3,0.1

Type RM Length L Ch R = 1 ,10001   ,492.4,499,503.5
XS GIS Cut Line= 6
1679776.95429026434034.3320324271679957.75970292434047.020327255
1680132.33021992434059.2706308361680207.14634326434064.520620346
1680294.40830784434070.9792688341680386.53476401434099.237086341
#Sta/Elev= 30
       0 1141.62    23.2 1127.79    79.4 1108.03   115.4 1084.31   131.5 1077.23
   162.4 1057.84   171.6 1055.16   177.4  1051.7   195.6 1037.75   203.7 1033.51
   215.7 1023.66   231.7 1014.74   239.7 1006.79   251.8 1003.69   271.8  991.49
   291.9  985.26   295.9  984.55  312.67985.2778     328  987.56   444.3  990.22
   476.3  995.54   496.4  995.54   500.4  998.37   516.5 1018.22   527.8 1025.95
   551.3 1046.34     563 1054.22   575.8 1057.86   591.4 1068.29   615.1 1080.14
#Mann= 5, -1 ,  0
       0     0.1       0   291.9   0.045       0  312.67     0.1       0
  471.25    0.06       0  578.75     0.1       0
Bank Sta=291.9,312.67
XS Rating Curve= 0 ,0
Exp/Cntr(USF)=0,0
Exp/Cntr=0.3,0.1

Type RM Length L Ch R = 1 ,9502    ,502.9,501.1,489.9
XS GIS Cut Line= 6
1679585.86641784434294.2137304991679736.20207517434395.459919095
1679881.35368776434493.2149729281679943.49988893434535.622696504
1680016.35735476434587.9598621731680106.13014109434635.775711417
#Sta/Elev= 30
       0 1178.06    12.4 1169.51    37.9 1159.21    54.3 1150.85    89.7  1123.3
   118.5 1110.35   137.7  1092.8   147.4 1085.56   171.5 1075.03   190.8 1062.37
   202.1 1057.45   211.8  1049.5   224.5 1041.78   276.3  992.81   291.5  983.52
   294.4     983   311.4  982.49   323.2  982.97   383.7  985.22   461.8  984.33
   476.6  989.55   501.4   989.6   506.1  992.01   520.9  1007.9   530.3 1015.31
   556.5 1027.97   588.9  1050.1   607.2 1060.21     616  1066.6   622.9 1067.89
#Mann= 4, -1 ,  0
       0     0.1       0   294.4   0.045       0   323.2     0.1       0
  451.49    0.06       0
Bank Sta=294.4,323.2
XS Rating Curve= 0 ,0
Exp/Cntr(USF)=0,0
Exp/Cntr=0.3,0.1

Type RM Length L Ch R = 1 ,9001    ,496.8,499.3,501.7
XS GIS Cut Line= 5
1679497.80493392434823.139195802 1679869.6562046434898.875250846
1679943.03630717 434914.378500671680028.64702834434932.464750588
1680120.45786834434951.437153593
#Sta/Elev= 30
       0 1086.81     6.4 1079.48    26.9 1068.73    47.3 1051.69    63.6 1042.48
    75.8 1037.36    94.7 1026.36   121.8 1006.18   149.3  988.05   165.6   984.4
   194.2  982.09   263.6  980.06   304.4   981.8315.1154979.0608   328.9  977.46
339.6154 979.155   345.3  983.16   349.3  984.38   361.6  985.13   373.8  984.24
   379.6  985.64   386.1  991.19   398.4 1005.33   454.5 1048.14   512.8 1084.76
   555.1 1101.74   586.4 1112.67   602.7 1114.87     619 1122.28   635.7 1127.26
#Mann= 5, -1 ,  0
       0     0.1       0     270    0.06       0315.1154   0.045       0
339.6154    0.06       0  464.49     0.1       0
Bank Sta=315.1154,339.6154
XS Rating Curve= 0 ,0
Exp/Cntr(USF)=0,0
Exp/Cntr=0.3,0.1

Type RM Length L Ch R = 1 ,8502    ,497.5,499.8,499.3
XS GIS Cut Line= 6
1679384.95376192435250.9309771661679553.38912059435317.871788174
1679623.08648776435345.5721920881679785.71345909435410.204608753
1679867.02694476435442.5214732591679954.14881776 435477.14574784
#Sta/Elev= 30
       0 1113.57    37.8 1097.88    59.4 1081.34    80.9 1068.79    85.2 1064.97
    93.8 1052.49   106.7 1048.02   120.7 1038.25   126.9 1032.21   145.4 1009.41
   149.7 1005.06   171.3  988.19   184.2  980.45   192.8  977.98     210  976.81
   278.9  976.08     287  974.11   302.4  972.78   320.9  974.17   330.5  979.45
   336.3  981.29   395.1  982.78     408  986.37   437.6   989.7   472.6 1009.99
     507  1038.1   519.9 1041.96   541.4 1055.59     563 1063.72   612.5 1071.55
#Mann= 4, -1 ,  0
       0     0.1       0     287   0.045       0   320.9    0.06       0
  406.25     0.1       0
Bank Sta=287,320.9
XS Rating Curve= 0 ,0
Exp/Cntr(USF)=0,0
Exp/Cntr=0.3,0.1

Type RM Length L Ch R = 1 ,8002    ,496.6,502.2,505.1
BEGIN DESCRIPTION:
Structure 2 XS 4
END DESCRIPTION:
XS GIS Cut Line= 6
1679281.19773585435742.6652299171679373.14046533435771.743583843
 1679458.7196905435797.2218793331679529.11390667435824.683766678
1679617.16097467435872.0937768371679842.78257068435993.580082417
#Sta/Elev= 30
       0 1097.21    61.8 1070.11   107.9 1053.24   137.1 1038.64   166.3  1028.9
   170.5 1025.58   183.1 1010.47   191.5 1003.26   214.1  989.71   234.4  975.26
     243  973.33  293.88969.7188   301.8   968.6  320.98969.9374   328.3  974.87
   334.3  976.51   363.8  976.67   387.4  989.13   405.5  999.83   419.2 1013.56
   432.8 1024.93   478.2 1052.61   496.4 1067.73   514.6 1074.71     538 1092.14
   547.8 1097.51   564.5 1104.75   578.2 1105.77   591.2 1111.42   617.5 1132.66
#Mann= 4, -1 ,  0
       0     0.1       0  293.88   0.045       0  320.98    0.06       0
  506.28     0.1       0
Bank Sta=293.88,320.98
XS Rating Curve= 0 ,0
Exp/Cntr(USF)=0,0
Exp/Cntr=0.3,0.1

Type RM Length L Ch R = 1 ,7499    ,54.7,54.5,54.6
BEGIN DESCRIPTION:
Structure 2 XS 3
END DESCRIPTION:
XS GIS Cut Line= 6
1679003.30190429435968.6076914221679069.35557794436035.137742087
1679130.77146561436097.4624205831679183.31532378 436150.98003009
1679305.91809694436275.8541241741679432.89947028436405.188183084
#Sta/Elev= 30
       0 1070.28    23.9 1063.86    57.1 1052.78    74.1 1039.18    79.7  1038.9
    88.2 1043.58    93.8 1043.63   131.9 1028.85   150.4 1023.07   156.1 1019.28
   200.3  981.99   213.6  975.05   232.5  972.47   280.9  969.21   294.7  965.32
   303.2  964.35  318.35965.3125   328.6  967.78   387.4  972.75   409.8  972.71
   415.4  975.61   427.6  985.88   433.3  988.82   445.8  993.19   468.6 1003.55
   491.5 1009.48   533.1 1014.62     560 1019.57     600 1021.12   612.5 1020.18
#Mann= 5, -1 ,  0
       0     0.1       0  231.25    0.06       0   294.7   0.045       0
  318.35    0.06       0  376.25     0.1       0
Bank Sta=294.7,318.35
XS Rating Curve= 0 ,0
Exp/Cntr(USF)=0,0
Exp/Cntr=0.3,0.1

Type RM Length L Ch R = 1 ,7445    ,442.9,443,441.5
BEGIN DESCRIPTION:
Structure 2 XS 2
END DESCRIPTION:
XS GIS Cut Line= 6
1678971.13316772436013.5717741551679037.18684137 436080.10182482
1679098.60272904436142.4265033161679151.14658721436195.944112823
1679273.74936037436320.8182069071679400.73073371436450.152265817
#Sta/Elev= 30
       0 1044.57    35.5 1036.72    59.4 1025.72    66.2 1025.89    76.3  1029.8
      82 1030.19   126.4 1021.16   143.5 1014.79   149.9 1010.57   189.8  976.21
     201  975.57   229.1  970.03   274.8  968.51   289.3  964.82     297  964.22
   305.4  964.87   316.8   967.7     349   968.3     379  972.17   400.4  971.81
   406.1  976.02   419.6  990.33   430.9  998.27   442.1 1007.93   458.2 1019.23
   463.8 1021.97   491.7  1031.9   511.9 1040.61   531.7 1046.17   612.5 1060.49
#Mann= 5, -1 ,  0
       0     0.1       0  286.25    0.06       0   289.3   0.045       0
   305.4    0.06       0  426.25     0.1       0
Bank Sta=289.3,305.4
XS Rating Curve= 0 ,0
Exp/Cntr(USF)=0,0
Exp/Cntr=0.3,0.1

Type RM Length L Ch R = 1 ,7002    ,505.9,501.1,489.7
BEGIN DESCRIPTION:
Structure 2 XS 1
END DESCRIPTION:
XS GIS Cut Line= 6
1678658.45587109436391.7472650861678742.64730376436436.897765338
1678818.50312318436482.849117011 1678876.9452635436529.910702676
1679076.25031109436700.7433662561679155.79345909436751.924038172
#Sta/Elev= 30
       0  1091.7    15.5 1084.29    29.1 1080.85    56.3 1057.93      70 1052.31
      79 1046.24    83.6 1042.08    94.8 1026.33   106.6 1015.44   125.5 1006.59
     158   983.9     175  974.67   193.3  967.54   201.7  965.94   274.7   965.1
   300.2  961.61   300.2   961.6   316.1  961.08   321.4  961.68   334.3  969.58
   359.8  969.22   363.5  971.61   379.3  988.78   416.2 1008.35   439.2 1017.05
     479 1026.55   510.2 1038.66   545.4 1056.43   576.5 1065.93   616.3 1088.36
#Mann= 5, -1 ,  0
       0     0.1       0  259.26    0.06       0   300.2   0.045       0
   321.4    0.06       0  409.26     0.1       0
Bank Sta=300.2,321.4
XS Rating Curve= 0 ,0
Exp/Cntr(USF)=0,0
Exp/Cntr=0.3,0.1

Type RM Length L Ch R = 1 ,6501    ,485.6,498.7,522.5
XS GIS Cut Line= 6
1678532.60605717436982.2382100821678629.32338342437010.248980835
1678721.56663726437024.6367473451678801.25512618437031.161012501
1678902.57775818437031.5914578441679158.82757376437031.591457844
#Sta/Elev= 30
       0 1075.07    16.1 1068.16    45.3 1052.53    66.1 1044.74   101.6 1024.77
   123.8 1014.59   152.1 1006.31   196.3  983.75   222.3  977.07     252  964.75
   268.8  962.01   296.9  961.64   308.9  960.33   316.9  957.74   328.9  957.07
   344.9  957.77   348.9  958.72   360.9  966.69   376.9  968.53   392.9  968.07
   424.9  993.63   447.9 1005.64   463.9 1010.98   480.9  1019.9   496.9 1032.02
   508.9 1047.58   540.9 1064.22   564.9 1081.88   604.9 1099.07   631.6 1113.29
#Mann= 4, -1 ,  0
       0     0.1       0   316.9   0.045       0   344.9    0.06       0
  445.33     0.1       0
Bank Sta=316.9,344.9
XS Rating Curve= 0 ,0
Exp/Cntr(USF)=0,0
Exp/Cntr=0.3,0.1

Type RM Length L Ch R = 1 ,6002    ,503.4,500.1,487.8
XS GIS Cut Line= 6
1678469.94345284437046.1206282531678503.99850284437138.013817176
1678513.98273484437225.1652176681678517.20549743437300.096170172
 1678524.7254955437474.9344031661678532.51452193437656.016718179
#Sta/Elev= 30
       0 1062.37    19.1 1052.83    53.8  1038.7    92.2 1020.62   100.5  1015.4
   129.3 1005.71   156.9  984.42   197.1  958.46   205.1  956.72   269.2   957.2
   301.2  954.01   313.2  953.52  322.45954.0833   333.2  961.49   337.2  962.76
   361.3  963.56   373.3  971.77   385.3   973.2   393.3  976.18   404.6  987.25
   413.3  998.63   441.3 1020.21   453.3 1034.69   457.3 1037.69   493.4 1051.04
   525.4 1072.25   561.4    1084   577.5 1094.44   589.5 1096.73     617 1113.31
#Mann= 5, -1 ,  0
       0     0.1       0   301.2   0.045       0  322.45     0.1       0
  380.72    0.06       0  475.72     0.1       0
Bank Sta=301.2,322.45
XS Rating Curve= 0 ,0
Exp/Cntr(USF)=0,0
Exp/Cntr=0.3,0.1

Type RM Length L Ch R = 1 ,5502    ,512.4,501.3,485.4
XS GIS Cut Line= 6
1677847.30395009437096.5188214181677907.81596817437168.124321252
 1678077.2503406437368.619327083  1678120.216462 437430.50371775
1678147.75019959437520.3585249191678170.78591467437622.960353836
#Sta/Elev= 30
       0 1088.34      21 1090.39    32.2 1089.93    68.1 1084.34   125.5 1064.74
   151.9 1045.35   170.9 1035.41   187.2 1017.65     220   997.8   236.7  981.38
   261.9  960.66   272.3  955.11   287.3  954.64   298.5  950.05   312.8  949.21
   321.3  950.01   340.4  952.57   375.6   952.6   395.1  957.99   419.5  956.86
   450.4  981.93   468.4  991.23   479.7  998.68   500.7 1005.32   513.2 1006.16
   521.6 1008.74   546.5 1020.95   570.8 1037.12   595.4 1048.07   630.7 1069.03
#Mann= 5, -1 ,  0
       0     0.1       0   298.5   0.045       0   321.3     0.1       0
  366.25    0.06       0  416.25     0.1       0
Bank Sta=298.5,321.3
XS Rating Curve= 0 ,0
Exp/Cntr(USF)=0,0
Exp/Cntr=0.3,0.1

Type RM Length L Ch R = 1 ,5001    ,476.6,507,515.4
XS GIS Cut Line= 6
1677444.08625259437683.8575417551677624.84606168 437697.17674084
 1677799.3729436437710.0379355851677874.17003809437715.549407512
1677961.43364309437721.9801689241678053.72512518437745.221920341
#Sta/Elev= 30
       0 1113.56       8 1109.76    20.1 1093.82    44.1 1082.68    60.2 1073.12
    92.3 1061.87   116.3 1046.23   156.5 1023.03   172.5 1011.75   196.6 1000.66
   212.6  998.51   244.7  988.29   256.7  979.54   262.2  974.02   272.8  960.34
   280.8  952.67  288.02947.9293   296.8  946.48     324  947.73   336.9  948.09
   351.8  951.66   421.2  955.05   437.7  961.63   465.3  961.56   505.4  990.25
   546.3 1003.73   562.8 1011.21     571 1016.23   591.6 1032.94   613.9  1042.7
#Mann= 5, -1 ,  0
       0     0.1       0  288.02   0.045       0     324     0.1       0
  451.25    0.06       0  548.75     0.1       0
Bank Sta=288.02,324
XS Rating Curve= 0 ,0
Exp/Cntr(USF)=0,0
Exp/Cntr=0.3,0.1

Type RM Length L Ch R = 1 ,4494    ,508.5,492.2,481.7
XS GIS Cut Line= 6
1677451.91924217437950.2749879211677645.11964317438032.844376594
  1677715.650342438086.0007663371677733.22839084438185.781406671
1677763.16271417438258.313741922   1677860.31147 438422.75271751
#Sta/Elev= 30
       0 1070.35    31.4 1052.57      56 1035.59      86 1020.08   107.5 1006.65
   142.8  991.85   160.5  990.37     187  981.86   209.1  980.85     244  971.94
   279.1  959.54   305.2  957.41   317.4  952.64   329.6  943.47   349.9  941.26
  359.35943.4788   362.1  944.78   374.2  956.81   378.3  958.59   398.6  960.68
   465.5  962.06   486.6  970.01   508.1  983.39   545.7  995.22   575.2 1002.48
   600.2 1017.82   609.7 1028.71     624 1039.66     647 1066.38   669.5 1087.36
#Mann= 5, -1 ,  0
       0     0.1       0  318.55    0.06       0   329.6   0.045       0
  359.35    0.06       0  538.34     0.1       0
Bank Sta=329.6,359.35
XS Rating Curve= 0 ,0
Exp/Cntr(USF)=0,0
Exp/Cntr=0.3,0.1

Type RM Length L Ch R = 1 ,4002    ,497.4,501,499.7
XS GIS Cut Line= 6
1677180.16125551438334.8808460091677246.13061176438405.585429013
1677318.61898383438455.4032427521677473.73022218438536.430639759
1677539.08442217438573.3052379191677695.40924075438665.508137509
#Sta/Elev= 30
       0 1082.63    18.7 1077.08    58.6 1054.59    67.9 1044.09    80.4 1026.84
    95.3 1010.77   103.1  998.87   108.8  995.39   167.1  976.85   199.9  957.03
     234  953.12   272.1  951.71   285.6  944.37   293.3  937.33   299.2  935.97
   325.3  937.27   362.4  940.13     385  950.21   412.9  950.97   417.3  954.84
   426.1  969.43   433.1  975.01   454.4   984.7   484.6  992.33   505.1   999.8
   519.3 1008.42   533.3 1020.37   561.2 1032.36   593.7 1056.16   616.2  1068.8
#Mann= 5, -1 ,  0
       0     0.1       0   293.3   0.045       0   325.3     0.1       0
  389.66    0.06       0   494.7     0.1       0
Bank Sta=293.3,325.3
XS Rating Curve= 0 ,0
Exp/Cntr(USF)=0,0
Exp/Cntr=0.3,0.1

Type RM Length L Ch R = 1 ,3501    ,568.1,562.4,551.6
XS GIS Cut Line= 6
1676773.47145209438572.2055025851676981.99662559438721.631384835
1677067.18772817438774.1640881751677128.57376026438820.850674585
1677198.06837192438884.6120299991677271.46783142438961.667650178
#Sta/Elev= 30
       0 1033.29    41.8 1028.04    85.3 1019.52   101.7  1014.6     131 1001.07
   160.7  994.45   174.1  987.76   185.6  985.54   199.9  976.21   214.3  970.68
   231.5  957.69   249.3  948.25   254.7   946.3   277.8  944.74   283.4  941.39
   292.6  931.23   301.3  930.09   324.1  931.15   338.9  933.71   381.8  934.86
   398.9  944.33   423.1  944.55   433.2  951.33     487  959.47   509.1  965.87
     531  977.48   569.1   987.5   588.9  994.49   605.3 1006.17   634.5 1035.17
#Mann= 6, -1 ,  0
       0    0.06       0  163.76     0.1       0  286.54    0.06       0
   292.6   0.045       0   324.1    0.06       0  396.62     0.1       0
Bank Sta=292.6,324.1
XS Rating Curve= 0 ,0
Exp/Cntr(USF)=0,0
Exp/Cntr=0.3,0.1

Type RM Length L Ch R = 1 ,2938    ,192.2,203.6,217.6
BEGIN DESCRIPTION:
Structure 1 XS 4
END DESCRIPTION:
XS GIS Cut Line= 5
1676617.64532018439314.0402236511676711.39546075439301.161968567
1676798.89528576439290.0540511541676873.89546384439285.456291311
1677230.14540751439285.456291311
#Sta/Elev= 30
       0 1071.73     6.5    1068    26.7 1050.61    46.9 1038.32      55 1035.67
    79.2 1009.86   107.5  983.71   147.8  964.99   167.9  949.66   184.1  943.37
   216.1  943.38   236.2  931.21   248.2  927.78   272.2  927.62   295.3   924.1
   300.2  923.53   320.2  924.22   332.2  930.37   344.2   931.7   360.2  930.77
   400.2   943.6   428.2  961.68   460.2  970.06   483.3  979.44   504.2  991.95
   520.2   997.6   532.2 1008.72   540.2 1013.99   571.3  1025.6   614.2 1048.65
#Mann= 5, -1 ,  0
       0     0.1       0  287.97    0.06       0   295.3   0.045       0
   320.2    0.06       0  387.97     0.1       0
Bank Sta=295.3,320.2
XS Rating Curve= 0 ,0
Exp/Cntr(USF)=0,0
Exp/Cntr=0.3,0.1

Type RM Length L Ch R = 1 ,2735    ,54.7,52.1,53.6
BEGIN DESCRIPTION:
Structure 1 XS 3
END DESCRIPTION:
XS GIS Cut Line= 6
1676630.75652681439393.9209846111676840.75161135439415.432676198
1676855.09273908439450.2611292441676867.38513427439468.699722034
1676942.16387169439539.3809943921677226.93769366439534.259163061
#Sta/Elev= 30
       0 1053.08     9.4 1047.08    25.5 1040.94    33.5 1034.66    65.7 1002.56
    77.8  987.23    81.8  983.88    97.9  973.66   110.6  967.95   150.1  945.74
   166.2  941.61   178.3  934.46     254  931.39  275.68922.1829   288.4  921.25
   313.8  922.11   321.5  923.33   327.9  927.44   334.7   929.1   407.8  928.93
   435.8  953.16   455.8  965.49   504.3   983.1   535.9  990.72   547.8  998.15
   579.8  1025.2   599.8 1039.27   615.8 1048.25   643.8 1059.67   658.6 1067.49
#Mann= 5, -1 ,  0
       0     0.1       0  275.68   0.045       0   313.8     0.1       0
  433.82    0.06       0  533.82     0.1       0
Bank Sta=275.68,313.8
XS Rating Curve= 0 ,0
Exp/Cntr(USF)=0,0
Exp/Cntr=0.3,0.1

Type RM Length L Ch R = 1 ,2683    ,297.2,289,267.4
BEGIN DESCRIPTION:
Structure 1 XS 2
END DESCRIPTION:
XS GIS Cut Line= 6
1676634.85399188439417.4814087311676801.82569324439448.212396712
1676849.97090775439516.8449365381676909.38415118439560.892685979
1676943.18823796439582.4043775661677223.86459486439571.136348639
#Sta/Elev= 30
       0 1043.51    21.6 1032.63      42 1019.12    65.5  992.51    78.6  981.35
    94.8  976.02   131.4  951.27   155.8  939.58   174.5  933.54   250.4   931.6
   263.5  923.48  268.41921.7197   291.1  920.99   311.1  921.71   335.5  927.64
   372.6  929.15   400.6  928.54   404.6  929.88   420.4  940.41   440.6  960.06
   448.6  965.79   496.7  983.57   508.7  985.97   520.7  992.89   540.7   999.4
   556.7 1011.09   588.7 1038.73   604.8 1048.18   616.8 1052.34   648.5 1068.51
#Mann= 7, -1 ,  0
       0     0.1       0  268.41   0.045       0   311.1     0.1       0
  367.57    0.06       0  427.64     0.1       0  447.64    0.06       0
  527.64     0.1       0
Bank Sta=268.41,311.1
XS Rating Curve= 0 ,0
Exp/Cntr(USF)=0,0
Exp/Cntr=0.3,0.1

Type RM Length L Ch R = 1 ,2394    ,391,392.8,394.5
BEGIN DESCRIPTION:
Structure 1 XS 1
END DESCRIPTION:
XS GIS Cut Line= 6
1676646.51967088439877.7315287411676737.59363572439852.227314663
1676823.33493405 439832.011147751676896.93682098439816.497071159
 1677156.4750158439777.1759555761677248.77371571439760.535896999
#Sta/Elev= 30
       0 1040.18    18.5 1032.63      39 1020.54    50.9 1009.03    68.1  995.93
    76.4  984.96    88.9  975.29    99.7  969.74   121.8  962.03     167  931.38
   195.7  926.94   281.7  924.04   311.4919.7704   321.8  919.27   342.8  919.78
     359  929.22   390.6  930.27   398.7  938.24   406.7  956.47   411.7  963.31
   422.9  968.84   439.1  974.37   451.2  976.48   463.4  982.33   471.5  987.79
   491.7 1005.99     520 1021.27   543.9 1039.81   569.1 1051.61   614.2 1079.55
#Mann= 5, -1 ,  0
       0     0.1       0  267.89    0.06       0   311.4   0.045       0
   342.8    0.06       0  462.89     0.1       0
Bank Sta=311.4,342.8
XS Rating Curve= 0 ,0
Exp/Cntr(USF)=0,0
Exp/Cntr=0.3,0.1

Type RM Length L Ch R = 1 ,2001    ,494.1,497.3,504.5
XS GIS Cut Line= 5
1676765.88419692440174.4713269171677122.13446867440174.471326917
1677197.13431868440181.000513345 1677284.6295505440191.210794762
1677378.18546575440203.426321507
#Sta/Elev= 30
       0 1062.41    14.2 1049.72    26.2 1042.25    42.2 1029.26    86.2  998.15
    90.2  994.19    98.2  982.35   106.2  976.52   138.2  965.49   150.2  963.03
   174.2  950.02   202.2  932.13   210.2  928.95   230.2  925.86   242.2  919.98
   286.2  918.09   292.2  916.44   306.2  915.75   320.2  916.45   338.2  921.05
   435.5  921.05   446.6  924.94   474.8  940.16   486.9  942.31     511  942.46
   519.1  945.46   539.3   958.5   554.6  964.05   587.7  971.45     614  974.91
#Mann= 5, -1 ,  0
       0     0.1       0   292.2   0.045       0   320.2     0.1       0
  431.53    0.07       0  539.62    0.06       0
Bank Sta=292.2,320.2
XS Rating Curve= 0 ,0
Exp/Cntr(USF)=0,0
Exp/Cntr=0.3,0.1
